--- Sevenmile_Creek_FINAL.prj (project) ---

Proj Title=Sevenmile Creek
Current Plan=p02
Default Exp/Contr=0.3,0.1
English Units
Geom File=g01
Flow File=f02
Plan File=p02
Y Axis Title=Elevation
X Axis Title(PF)=Main Channel Distance
X Axis Title(XS)=Station
BEGIN DESCRIPTION:
####(Watershed Name)####
SEVENMILE CREEK
HCFCD Unit X###-##-##
(Flood Hazard, Floodway) Model
10, 2, 1, 0.2% Event
Filename:  n:\NC_flood\60138\Orange\URS\Limited_Detail\ENG\Sevenmile Creek\Sevenmile Creek.prj
Prepared by:  ________     Date: ________
Reviewed by:  ________     Date: ________
STATUS (Draft RAS, SVSQ, FINAL)
END DESCRIPTION:
DSS Export Rating Curves= 0
DSS Export Rating Curve Sorted= 0
DSS Export Volume Flow Curves= 0
DXF OffsetX= 0
DXF OffsetY= 0
DXF ScaleX= 1
DXF ScaleY= 10

--- Sevenmile_Creek_FINAL.p02 (plan) ---

Plan Title=floodway
Version=Version 3.0.1  Mar 2001
Short Identifier=fw
Geom File=g01
Flow File=f02
Subcritical Flow
K Sum by GR= 0
Std Step Tol= 0.01
Critical Tol= 0.01
Num of Std Step Trials= 20
Max Error Tol= 0.3
Flow Tol Ratio= 0.001
Split Flow NTrial= 30
Split Flow Tol= 0.02
Split Flow Ratio= 0.02
Log Output Level= 0
Friction Slope Method= 1
Unsteady Friction Slope Method= 2
Parabolic Critical Depth
Global Vel Dist= 0 , 0 , 0
Global Log Level= 0
CheckData=True
Encroach Param=-1 ,0,0, 2
Encroach River=Sevenmile Creek
Encroach Reach=Reach - 1
Encroach Node=36464.3
       1    4871    5013
Encroach Node=35934.7
       1 4989.01 5009.48
Encroach Node=35684.0
       1 4958.22  5084.2
Encroach Node=34756.4
       1    4985    5040
Encroach Node=34120.5
       1 4920.04 5123.17
Encroach Node=33790.9
       1 4938.58 5084.75
Encroach Node=33202.6
       1 4928.12 5041.12
Encroach Node=32675.6
       1 4950.94 5070.98
Encroach Node=31975.6
       1    4824    5012
Encroach Node=31050.2
       1    4929    5015
Encroach Node=30409.1
       1 4825.66 5024.25
Encroach Node=29930.5
       1 4969.01 5081.91
Encroach Node=29500.0
       1 4937.92 5099.14
Encroach Node=29000.0
       1 4940.86 5125.84
Encroach Node=28388.9
       1 4881.34 5054.18
Encroach Node=28012.1
       1  4910.8 5081.78
Encroach Node=27500.0
       1 4881.77 5024.84
Encroach Node=27150.3
       1 4939.81 5089.89
Encroach Node=26669.0
       1 4908.07 5036.57
Encroach Node=25716.7
       1 4887.36    5010
Encroach Node=25413.3
       1    4835    5020
Encroach Node=24555.3
       1 4972.52  5053.1
Encroach Node=24131.7
       1  4939.2 5062.48
Encroach Node=23748.9
       1  4970.4 5075.43
Encroach Node=23000.0
       1    4945    5020
Encroach Node=22528.7
       1    4960 5047.19
Encroach Node=21679.4
       1    4905    5018
Encroach Node=21135.7
       1 4944.85 5055.05
Encroach Node=21112.9
       1 4944.85 5055.05
Encroach Node=21090.2
       1 4944.85 5055.05
Encroach Node=20701.0
       1 4945.09 5030.65
Encroach Node=19998.9
       1  4963.4 5017.15
Encroach Node=19407.7
       1 4714.38 5032.81
Encroach Node=18869.5
       1 4934.18 5018.63
Encroach Node=18436.5
       1 4987.77 5051.48
Encroach Node=18066.4
       1    4980    5083
Encroach Node=17606.3
       1    4980    5145
Encroach Node=17000.0
       1 4984.81    5053
Encroach Node=16710.2
       1 4973.35 5024.63
Encroach Node=16384.5
       1 4730.12 5023.32
Encroach Node=15618.8
       1    4975    5358
Encroach Node=14887.1
       1 4880.76 5079.92
Encroach Node=14540.3
       1    4980    5055
Encroach Node=14098.1
       1    4845    5020
Encroach Node=13425.2
       1 4945.97 5035.53
Encroach Node=12949.0
       1 4977.81 5034.96
Encroach Node=12589.7
       1  4979.5 5151.92
Encroach Node=11924.3
       1    4919    5013
Encroach Node=11410.1
       1 4945.56 5032.65
Encroach Node=10966.0
       1  4983.3 5039.67
Encroach Node=10504.4
       1 4975.01 5038.71
Encroach Node=9896.9
       1 4897.79 5034.65
Encroach Node=9206.8
       1  4971.4 5074.59
Encroach Node=8839.6
       1 4952.94  5089.5
Encroach Node=8442.9
       1 4915.12 5036.65
Encroach Node=7955.6
       1    4747    5017
Encroach Node=7534.1
       1    4715    5020
Encroach Node=7067.5
       1    4872    5128
Computation Interval=1HOUR
Output Interval=1HOUR
Run HTab= 0
Run UNet= 0
Run PostProcess= 0
UNET Theta= 1
UNET ZTol= 0.02
UNET ZSATol= 0.1
UNET MxIter= 20
UNET MaxInSteps= 20
UNET DtIC= 0
UNET DtMin= 0
UNET MaxCRTS= 20
UNET WFStab= 2
UNET SFStab= 1
UNET WFX= 1
UNET SFX= 1
UNET Convert EG Bridges=-1
UNET Use Existing IB Tables=-1
Instantaneous Interval=1HOUR
Write IC File= 0
Write Velocity= 0
Write Detailed= 0

--- Sevenmile_Creek_FINAL.f02 (steady flow) ---

Flow Title=100 Year floodway
Version=Version 3.0.1  Mar 2001
Number of Profiles= 2
Profile Names=100-Year,100 yr fw
River Rch & RM=Sevenmile Creek,Reach - 1       ,36464.3
     764     764
River Rch & RM=Sevenmile Creek,Reach - 1       ,34120.5
    1510    1510
River Rch & RM=Sevenmile Creek,Reach - 1       ,27500
    2995    2995
River Rch & RM=Sevenmile Creek,Reach - 1       ,18869.5
    3184    3184
River Rch & RM=Sevenmile Creek,Reach - 1       ,11410.1
    3920    3920
Boundary for River Rch & Prof#=Sevenmile Creek,Reach - 1       , 1
Up Type= 0
Dn Type= 1
Dn Known WS=532.7
Boundary for River Rch & Prof#=Sevenmile Creek,Reach - 1       , 2
Up Type= 0
Dn Type= 1
Dn Known WS=533.4
DSS Import GetInterval= 0
DSS Import GetPeak= 0
DSS Import FillOption= 0

--- Sevenmile_Creek_FINAL.g01 (geometry) ---

Geom Title=Geom 01 by CodeH2 for Windows

River Reach=Sevenmile Creek,Reach - 1
Reach XY= 30
 1940233.4167027 837113.09628810      1942680.29       838383.08
      1943197.54       839183.85      1943413.37        839035.7
      1943924.23       839356.26      1946444.22       841985.39
      1947048.83       841759.96      1947231.26        842115.7
      1948441.14       842678.61      1949208.64       842795.89
      1949624.38       842325.26      1950002.85       842876.68
      1950557.94       842941.83      1951236.76       842371.13
      1952039.38       842620.24      1952044.59       843145.63
      1952647.12       843511.52      1953094.33       842651.51
      1953304.38       842916.29      1953620.24       842793.28
      1953312.53       842273.89      1953645.36       841748.98
      1954605.16        841665.3      1954761.11       840609.14
      1955043.49       841231.83      1955751.95       840830.42
      1955950.94       841086.59      1955747.95        841907.7
       1956639.4       842048.37 1957179.7742462 842741.80367615

Type RM Length L Ch R = 1 ,36464.3,529.6,529.6,529.6
XS GIS Cut Line= 3
 1940027.6936689 837465.47737028 1940229.4073466 837120.17090507
 1940293.1604162 837006.83211455
BEGIN DESCRIPTION:
Sevenmile Creek 73.0
END DESCRIPTION:
#Sta/Elev= 24
    4592  629.79    4612  627.29    4622  625.55    4642  623.82    4652   623.6
    4662  623.02    4712  621.41    4842   620.8    4852  620.21    4862  619.16
    4882  620.61    4902  619.73    4932   621.1    4942  621.16    4952  621.57
    4962  621.62  4991.9  618.98    4996  618.44  4997.5  615.44  5002.5  615.44
    5004  618.44  5011.9   620.4  5081.9  630.02  5121.9  637.06
#Mann= 3 , 1 , 0
 4592.00    0.11       0    4996    0.04       0    5004    0.11       0
Bank Sta=4996.00,5004.00
Exp/Cntr=0.3,0.1

Type RM Length L Ch R = 1 ,35934.7,250.7,250.7,250.7
XS GIS Cut Line= 3
 1940501.9543491 837530.41626467 1940578.1326877 837421.03198366
 1940691.2001721 837209.33116173
BEGIN DESCRIPTION:
Sevenmile Creek 72.0
END DESCRIPTION:
#Sta/Elev= 23
  4865.2  629.46  4915.2  622.28  4935.2  620.12  4945.2   618.7  4955.2  618.71
  4965.2  618.26  4975.2  617.36  4985.2  616.03  4995.2  614.05    4996  613.16
  4997.5  610.16  5002.5  610.16    5004  613.16  5008.5  615.41  5018.5  617.22
  5038.5  617.83  5048.5  618.42  5148.5  619.66  5158.5  620.14  5168.5  621.64
  5188.5   625.8  5208.5  628.25  5238.5  633.23
#Mann= 3 , 1 , 0
 4865.20    0.11       0    4996    0.04       0    5004    0.11       0
Bank Sta=4996.00,5004.00
Exp/Cntr=0.3,0.1

Type RM Length L Ch R = 1 ,35684.0,927.6,927.6,927.6
XS GIS Cut Line= 3
 1940660.6006405 837671.21359607 1940769.5897377 837530.43601224
 1940894.0635196 837325.16345959
BEGIN DESCRIPTION:
Sevenmile Creek 71.0
END DESCRIPTION:
#Sta/Elev= 26
  4818.6  631.94  4858.6  627.33  4868.6  625.91  4878.6  624.15  4898.6  620.19
  4938.6  615.67  4948.6     616  4958.6  615.18  4968.6  616.68  4978.6   617.1
  4988.6  617.07    4996  612.52  4997.5  609.52  5002.5  609.52    5004  612.52
  5006.7  615.12  5016.7  616.15  5026.7  616.29  5046.7  615.67  5056.7  615.98
  5066.7  615.39  5076.7  615.15  5086.7  615.37  5096.7  615.97  5186.7  619.34
  5236.7  629.66
#Mann= 3 , 1 , 0
 4818.60    0.11       0    4996    0.04       0    5004    0.11       0
Bank Sta=4996.00,5004.00
Exp/Cntr=0.3,0.1

Type RM Length L Ch R = 1 ,34756.4,635.9,635.9,635.9
XS GIS Cut Line= 3
 1941179.8548449 837964.63325067 1941279.0022458 837793.68945601
 1941422.2140330 837553.09365344
BEGIN DESCRIPTION:
Sevenmile Creek 69.0
END DESCRIPTION:
#Sta/Elev= 30
  4806.2  626.63  4876.2  624.46  4886.2  623.68  4966.2  614.34  4976.2  613.49
  4986.2  613.17    4996  610.14  4997.5  607.14  5002.5  607.14    5004  610.14
  5013.8  613.89  5043.8  612.86  5053.8  612.77  5073.8  613.63  5083.8  613.26
  5093.8  613.36  5103.8  613.85  5113.8  613.55  5153.8  614.18  5163.8  613.58
  5173.8  613.68  5183.8  614.29  5193.8  614.17  5203.8  614.33  5213.8  614.92
  5223.8   615.9  5233.8  616.41  5253.8   619.4  5273.8  624.06  5283.8  625.96
#Mann= 3 , 1 , 0
 4806.20    0.11       0    4996    0.04       0    5004    0.11       0
Bank Sta=4996.00,5004.00
Exp/Cntr=0.3,0.1

Type RM Length L Ch R = 1 ,34120.5,329.6,329.6,329.6
XS GIS Cut Line= 3
 1941679.0107253 838145.83367301 1941781.5770021 837964.63325067
 1941894.4948243 837787.62693473
BEGIN DESCRIPTION:
Sevenmile Creek 68.0
END DESCRIPTION:
#Sta/Elev= 24
  4792.2  624.96  4832.2  621.28  4862.2  617.28  4892.2  610.07  4902.2  608.74
  4932.2  609.62  4952.2  609.12  4972.2  609.67  4982.2  609.52  4992.2   608.8
  4995.6  608.14  4997.1  605.14  5002.8  605.14  5004.3  608.14  5010.4  608.29
  5020.4  609.44  5030.4  609.65  5120.4   608.7  5140.4  609.21  5150.4  609.82
  5170.4  613.65  5180.4  616.96  5190.4  620.64  5210.4  625.67
#Mann= 3 , 1 , 0
 4792.20    0.14       0  4995.6    0.04       0  5004.3    0.14       0
Bank Sta=4995.60,5004.30
Exp/Cntr=0.3,0.1

Type RM Length L Ch R = 1 ,33790.9,588.3,588.3,588.3
XS GIS Cut Line= 3
 1941921.7509137 838268.91320516 1942034.5738181 838087.71278282
 1942136.4680996 837939.23825837
BEGIN DESCRIPTION:
Sevenmile Creek 67.0
END DESCRIPTION:
#Sta/Elev= 20
  4794.5   621.7  4824.5  618.62  4884.5  610.37  4924.5  608.45  4934.5  608.28
  4964.5  608.57  4994.5  607.36  4995.7  606.69  4997.2  603.69  5002.9  603.69
  5004.4  606.69  5004.5  607.23    5008  607.29    5048  608.25    5058     608
    5068  608.18    5098   607.8    5108  608.33    5168  621.05    5188  625.91
#Mann= 3 , 1 , 0
 4794.50    0.14       0  4995.7    0.04       0  5004.4    0.14       0
Bank Sta=4995.70,5004.40
Exp/Cntr=0.3,0.1

Type RM Length L Ch R = 1 ,33202.6,527,527,527
XS GIS Cut Line= 3
 1942260.2196271 838521.91002125 1942352.5292762 838385.15498552
 1942458.9275154 838215.78635979
BEGIN DESCRIPTION:
Sevenmile Creek 66.0
END DESCRIPTION:
#Sta/Elev= 18
    4832  613.22    4882  607.72    4902  605.95    4922   605.8    4932  605.21
    4972  603.72    4982  604.38    4992  603.72  4995.7  602.54  4997.2  599.54
  5002.8  599.54  5004.3  602.54    5007  603.92    5057  605.64    5067  606.45
    5107  612.93    5127  616.93    5197  627.42
#Mann= 3 , 1 , 0
 4832.00    0.14       0  4995.7    0.04       0  5004.3    0.14       0
Bank Sta=4995.70,5004.30
Exp/Cntr=0.3,0.1

Type RM Length L Ch R = 1 ,32675.6,700,700,700
XS GIS Cut Line= 3
 1942547.4052021 838682.59718823 1942680.7413619 838508.23451768
 1942783.8319394 838385.81445698
BEGIN DESCRIPTION:
Sevenmile Creek 65.0
END DESCRIPTION:
#Sta/Elev= 26
  4784.2  616.07  4814.2  612.85  4834.2  609.27  4854.2  606.79  4884.2  604.56
  4904.2  604.02  4964.2  601.88  4974.2  601.96  4984.2  602.34  4994.2  601.62
  4995.7  599.98  4997.2  596.98  5002.9  596.98  5004.4  599.98  5013.7  602.51
  5023.7  603.02  5043.7  602.79  5053.7  603.25  5083.7  602.58  5103.7  603.82
  5113.7  603.71  5123.7  604.51  5133.7  607.14  5143.7   610.2  5153.7  614.21
  5163.7  616.91
#Mann= 3 , 1 , 0
 4784.20    0.14       0  4995.7    0.04       0  5004.4    0.14       0
Bank Sta=4995.70,5004.40
Exp/Cntr=0.3,0.1

Type RM Length L Ch R = 1 ,31975.6,925.4,925.4,925.4
XS GIS Cut Line= 3
 1942859.6481214 839024.26015124 1943043.1422066 838771.48796145
 1943113.8598002 838687.30035002
BEGIN DESCRIPTION:
Sevenmile Creek 64.0
END DESCRIPTION:
#Sta/Elev= 30
  4686.1  613.76  4716.1  610.38  4726.1  608.72  4746.1   604.9  4756.1  603.29
  4766.1  602.11  4796.1  599.53  4816.1  597.49  4826.1  598.36  4856.1  599.71
  4876.1  599.44  4886.1  598.65  4906.1  598.57  4926.1  597.37  4936.1  598.08
  4946.1   599.1  4956.1  599.71  4976.1  600.07  4986.1  600.77  4995.7  596.74
  4997.2  593.74  5002.8  593.74  5004.3  596.74  5008.4  600.85  5018.4  601.51
  5028.4  602.75  5048.4  607.05  5058.4  608.59  5068.4  610.77  5108.4  617.53
#Mann= 3 , 1 , 0
 4686.10    0.14       0  4995.7    0.04       0  5004.3    0.14       0
Bank Sta=4995.70,5004.30
Exp/Cntr=0.3,0.1

Type RM Length L Ch R = 1 ,31050.2,641.1,641.1,641.1
XS GIS Cut Line= 3
 1943206.6953702 839413.42269570 1943426.0563066   839041.579157
 1943500.9652385 838877.82474784
BEGIN DESCRIPTION:
Sevenmile Creek 63.0
END DESCRIPTION:
#Sta/Elev= 30
  4569.6  612.44  4639.6  602.24  4649.6  601.74  4669.6  601.54  4699.6  599.52
  4709.6   599.8  4729.6  599.38  4739.6  598.75  4759.6  599.44  4779.6  599.54
  4789.6  598.89  4829.6  599.04  4899.6   597.2  4919.6  596.13  4939.6  596.68
  4979.6  596.38  4989.6  595.89  4995.7  592.37  4997.2  589.37  5002.9  589.37
  5004.4  592.37  5021.4  597.25  5031.4  598.72  5051.4  600.88  5081.4  602.76
  5101.4  605.57  5111.4  604.42  5121.4  604.63  5161.4  608.78  5181.4  610.24
#Mann= 3 , 1 , 0
 4569.60    0.14       0  4995.7    0.04       0  5004.4    0.14       0
Bank Sta=4995.70,5004.40
Exp/Cntr=0.3,0.1

Type RM Length L Ch R = 1 ,30409.1,478.6,478.6,478.6
XS GIS Cut Line= 3
 1943763.1200890 839667.95394925 1943918.3744353 839345.85911149
 1943973.1114468 839274.49313447
BEGIN DESCRIPTION:
Sevenmile Creek 61.0
END DESCRIPTION:
#Sta/Elev= 28
  4649.8  612.77  4689.8  606.75  4699.8  604.87  4729.8  599.98  4749.8  597.79
  4759.8  596.35  4769.8  595.17  4789.8  594.81  4809.8  593.82  4819.8  594.42
  4879.8  594.16  4899.8  594.48  4919.8  593.68  4939.8  593.89  4949.8  593.57
  4969.8  592.22  4989.8  592.44  4995.7  590.52  4997.2  587.52  5002.8  587.52
  5004.3  590.52  5007.3  590.87  5017.3  591.37  5047.3  593.99  5057.3  596.98
  5067.3  600.96  5077.3  604.66  5097.3  610.07
#Mann= 3 , 1 , 0
 4649.80    0.14       0  4995.7    0.04       0  5004.3    0.14       0
Bank Sta=4995.70,5004.30
Exp/Cntr=0.3,0.1

Type RM Length L Ch R = 1 ,29930.5,430.5,430.5,430.5
XS GIS Cut Line= 3
 1943998.7310156 839930.09108265  1944215.816638 839622.78805883
 1944320.8794479 839489.07175524
BEGIN DESCRIPTION:
Sevenmile Creek 60.0
END DESCRIPTION:
#Sta/Elev= 22
  4617.1  623.86  4807.1  605.66  4827.1  603.22  4837.1  602.34  4847.1  601.76
  4907.1  595.49  4927.1  594.27  4937.1  593.28  4947.1  592.69  4987.1  591.38
  4993.4  590.34  4995.7  590.04  4997.2  587.04  5002.8  587.04  5004.3  590.04
  5053.4  591.05  5063.4  591.73  5103.4  592.36  5113.4  593.22  5123.4   595.4
  5133.4  598.16  5163.4  611.01
#Mann= 3 , 1 , 0
 4617.10    0.14       0  4995.7    0.04       0  5004.3    0.14       0
Bank Sta=4995.70,5004.30
Exp/Cntr=0.3,0.1

Type RM Length L Ch R = 1 ,29500.0,500,500,500
XS GIS Cut Line= 3
 1944355.9535761 840063.00959236 1944524.9376017 839900.71095102
 1944769.6745326 839656.97681777
BEGIN DESCRIPTION:
Sevenmile Creek 59.0
END DESCRIPTION:
#Sta/Elev= 30
  4765.7  605.07  4775.7  603.67  4785.7  601.35  4795.7  600.66  4805.7  599.38
  4835.7  596.63  4885.7  592.73  4915.7  591.48  4935.7  589.79  4985.7  590.62
  4995.7  589.62  4997.2  586.62  5002.8  586.62  5004.3  589.62    5010  590.58
    5020  590.42    5030  590.84    5050  589.73    5080  589.96    5090  590.31
    5110  591.53    5140   591.3    5150  592.03    5160  593.41    5180  595.14
    5190  596.25    5220  600.48    5230  601.59    5240  602.42  5345.4  615.61
#Mann= 3 , 1 , 0
 4765.70    0.14       0  4995.7    0.04       0  5004.3    0.14       0
Bank Sta=4995.70,5004.30
Exp/Cntr=0.3,0.1

Type RM Length L Ch R = 1 ,29000.0,611.1,611.1,611.1
XS GIS Cut Line= 3
 1944670.8789031 840374.85633840 1944769.1371106 840280.25202685
 1945044.8681338 840033.52699616
BEGIN DESCRIPTION:
Sevenmile Creek 58.0
END DESCRIPTION:
#Sta/Elev= 30
  4863.6  603.96  4873.6  601.58  4893.6   595.2  4903.6  592.68  4913.6  590.66
  4933.6  587.36  4953.6  588.37  4963.6  587.75  4973.6  587.69  4983.6  588.58
  4993.6  587.78  4995.6   587.9  4997.1   584.9  5002.8   584.9  5004.3   587.9
    5010  588.34    5020  588.51    5030  588.29    5050  589.36    5120  589.69
    5140  590.23    5160  589.54    5180  590.94    5200  591.07    5260  592.58
    5270  593.88    5280  594.81    5300  596.13    5340  601.17    5370  606.97
#Mann= 3 , 1 , 0
 4863.60    0.14       0  4995.6    0.04       0  5004.3    0.14       0
Bank Sta=4995.60,5004.30
Exp/Cntr=0.3,0.1

Type RM Length L Ch R = 1 ,28388.9,376.8,376.8,376.8
XS GIS Cut Line= 3
 1945039.0035575 840729.16987613 1945234.6416541 840590.32993659
 1945396.9585560 840457.08471863
BEGIN DESCRIPTION:
Sevenmile Creek 57.0
END DESCRIPTION:
#Sta/Elev= 26
  4762.7  602.66  4772.7  601.29  4792.7  598.93  4802.7  597.26  4812.7  594.74
  4822.7  592.48  4842.7  589.39  4882.7  586.58  4902.7  586.75  4932.7  586.16
  4952.7  586.68  4962.7  586.48  4972.7  586.62  4992.7  585.15  4995.7  584.61
  4997.2  581.61  5002.9  581.61  5004.4  584.61  5032.6  585.61  5052.6  587.31
  5082.6  588.75  5102.6   589.1  5132.6  591.25  5142.6  592.47  5162.6  595.61
  5212.6   604.4
#Mann= 3 , 1 , 0
 4762.70    0.14       0  4995.7    0.04       0  5004.4    0.14       0
Bank Sta=4995.70,5004.40
Exp/Cntr=0.3,0.1

Type RM Length L Ch R = 1 ,28012.1,512.1,512.1,512.1
XS GIS Cut Line= 3
         1945175          841075 1945446.6119595 840898.02876697
 1945708.3927912 840713.91917105
BEGIN DESCRIPTION:
Sevenmile Creek 56.0
END DESCRIPTION:
#Sta/Elev= 30
  4670.8  598.09  4750.8   597.1  4770.8  597.99  4780.8  597.93  4850.8   592.8
  4860.8  591.78  4880.8  587.66  4930.8  585.75  4950.8  584.49  4970.8  584.57
  4980.8  585.18  4990.8  583.08    4995  582.54  4995.7  581.63  4997.2  578.63
  5002.8  578.63  5004.3  581.63    5005  581.87    5035     586    5075  586.69
    5095  587.95    5155  589.34    5165   589.9    5185  591.78    5195  592.13
    5205  592.08    5215   592.4    5235   593.8    5255  595.73    5315  604.15
#Mann= 3 , 1 , 0
 4670.80    0.14       0  4995.7    0.04       0  5004.3    0.14       0
Bank Sta=4995.70,5004.30
Exp/Cntr=0.3,0.1

Type RM Length L Ch R = 1 ,27500.0,349.7,349.7,349.7
XS GIS Cut Line= 3
 1945632.7027861 841563.84348238 1945808.4256303 841198.28320582
 1945851.4809969 841097.06149017
BEGIN DESCRIPTION:
Sevenmile Creek 55.0
END DESCRIPTION:
#Sta/Elev= 28
  4594.4  605.09  4644.4   600.9  4664.4  599.64  4694.4  595.42  4724.4  591.82
  4734.4  590.89  4744.4   590.4  4764.4  588.86  4774.4  588.36  4804.4  587.94
  4814.4  587.47  4824.4  587.36  4834.4  587.59  4844.4  587.57  4854.4   587.8
  4894.4   585.5  4904.4  584.52  4974.4  584.24  4984.4  583.95  4990.4  581.05
  4991.9  578.05  5008.1  578.05  5009.6  581.05    5030  583.13    5060  592.01
    5090  598.77    5100   600.4    5110  601.24
#Mann= 3 , 1 , 0
 4594.40    0.14       0  4990.4    0.04       0  5009.6    0.14       0
Bank Sta=4990.40,5009.60
Exp/Cntr=0.3,0.1

Type RM Length L Ch R = 1 ,27150.3,481.3,481.3,481.3
XS GIS Cut Line= 3
 1945800.3907770 841684.38467770 1945972.1615618 841467.20322565
 1946087.6425001 841316.32386553
BEGIN DESCRIPTION:
Sevenmile Creek 54.0
END DESCRIPTION:
#Sta/Elev= 30
  4720.8  600.96  4740.8  599.58  4750.8  598.54  4770.8  595.85  4800.8  593.52
  4810.8  592.29  4830.8  591.38  4850.8  589.02  4900.8  587.37  4920.8  584.96
  4930.8  584.05  4940.8  583.58  4960.8  583.67  4970.8  582.82  4990.4  580.11
  4991.9  577.11  5008.1  577.11  5009.6  580.11  5027.7  582.31  5047.7  582.11
  5057.7  583.59  5067.7  583.95  5097.7  584.49  5117.7  585.98  5127.7  587.04
  5137.7  589.55  5147.7  591.58  5167.7  596.46  5177.7  598.26  5187.7  600.56
#Mann= 3 , 1 , 0
 4720.80    0.14       0  4990.4    0.04       0  5009.6    0.14       0
Bank Sta=4990.40,5009.60
Exp/Cntr=0.3,0.1

Type RM Length L Ch R = 1 ,26669.0,952.3,952.3,952.3
XS GIS Cut Line= 3
 1946178.1660983 841947.56807150 1946318.4253122 841708.30235364
 1946367.0672135 841545.45772764
BEGIN DESCRIPTION:
Sevenmile Creek 53.0
END DESCRIPTION:
#Sta/Elev= 26
  4723.7  601.89  4753.7  599.27  4763.7  597.54  4783.7   595.5  4793.7  593.56
  4803.7  592.21  4813.7  591.21  4833.7  587.79  4843.7  586.97  4853.7  587.08
  4863.7   586.5  4873.7  585.51  4943.7  582.16  4973.7  582.35  4983.7  581.73
  4990.3   579.1  4991.8   576.1  5008.1   576.1  5009.6   579.1    5021  580.06
    5041  583.59    5061  584.88    5111  590.37    5131  593.08    5141   594.8
    5171  597.83
#Mann= 3 , 1 , 0
 4723.70    0.14       0  4990.3    0.04       0  5009.6    0.14       0
Bank Sta=4990.30,5009.60
Exp/Cntr=0.3,0.1

Type RM Length L Ch R = 1 ,25716.7,303.4,303.4,303.4
XS GIS Cut Line= 3
 1946756.1752856 842013.52699582 1946856.8982654  841738.2175177
 1946867.7528312 841669.01966060
BEGIN DESCRIPTION:
Sevenmile Creek 52.0
END DESCRIPTION:
#Sta/Elev= 24
  4697.2  598.66  4727.2  596.35  4747.2  595.32  4797.2  589.93  4807.2  588.27
  4817.2  586.94  4827.2  586.17  4847.2  584.03  4867.2  580.23  4877.2  580.28
  4887.2   581.6  4907.2  582.48  4917.2  582.44  4977.2  580.39  4987.2   579.4
  4990.3  577.18  4990.4  577.11  4991.9  574.11  5008.1  574.11  5009.6  577.11
  5010.4  586.75  5020.4  591.09  5040.4  596.87  5060.4  601.18
#Mann= 3 , 1 , 0
 4697.20    0.14       0  4990.3    0.04       0  5009.6    0.14       0
Bank Sta=4990.30,5009.60
Exp/Cntr=0.3,0.1

Type RM Length L Ch R = 1 ,25413.3,858,858,858
XS GIS Cut Line= 3
 1946943.6693356 842311.80232629 1947143.2291214 841806.59503556
 1947184.8189211 841672.91353680
BEGIN DESCRIPTION:
Sevenmile Creek 50.0
END DESCRIPTION:
#Sta/Elev= 30
  4459.2  597.61  4479.2  597.12  4519.2   593.5  4539.2  592.33  4559.2  592.03
  4569.2  591.01  4579.2  588.97  4619.2  586.24  4659.2  585.03  4739.2  584.39
  4749.2  583.79  4769.2  583.44  4789.2  581.86  4829.2   579.7  4839.2  580.12
  4859.2  579.46  4889.2   580.2  4969.2  580.42  4989.2  578.23  4990.4  576.23
  4991.9  573.23  5008.1  573.23  5009.6  576.23  5012.4  580.67  5052.4  584.92
  5082.4  588.88  5102.4   590.7  5112.4   592.2  5122.4  594.33  5142.4  599.74
#Mann= 3 , 1 , 0
 4459.20    0.11       0  4990.4   0.045       0  5009.6    0.14       0
Bank Sta=4990.40,5009.60
Exp/Cntr=0.3,0.1

Type RM Length L Ch R = 1 ,24555.3,423.6,423.6,423.6
XS GIS Cut Line= 3
 1947520.5232908 842546.30058066 1947591.3411848 842344.62353487
 1947661.3597630 842171.76516971
BEGIN DESCRIPTION:
Sevenmile Creek 49.0
END DESCRIPTION:
#Sta/Elev= 21
  4782.4  597.92  4812.4  595.28  4882.4  592.34  4902.4  590.89  4922.4  588.68
  4952.4   582.1  4962.4  580.29  4972.4  578.96  4990.4  575.33  4991.9  572.33
  5008.2  572.33  5009.7  575.33  5016.2  576.69  5026.2  578.57  5036.2  579.55
  5056.2   579.5  5066.2  580.17  5086.2     583  5116.2  588.11  5126.2  589.12
  5182.7  596.32
#Mann= 3 , 1 , 0
 4782.40    0.11       0  4990.4   0.045       0  5009.7    0.14       0
Bank Sta=4990.40,5009.70
Exp/Cntr=0.3,0.1

Type RM Length L Ch R = 1 ,24131.7,382.8,382.8,382.8
XS GIS Cut Line= 3
 1947880.1678202 842769.11116576 1947978.6314459 842506.54149716
 1948035.0988628 842346.24689442
BEGIN DESCRIPTION:
Sevenmile Creek 48.0
END DESCRIPTION:
#Sta/Elev= 24
  4718.5  599.81  4788.5  594.69  4808.5   593.8  4858.5  587.91  4898.5  581.86
  4908.5  580.71  4918.5  580.39  4928.5  580.44  4978.5  578.92  4988.5  578.25
  4990.4  574.78  4991.9  571.78  5008.1  571.78  5009.6  574.78  5028.9  578.68
  5048.9  578.54  5058.9  577.47  5068.9  578.08  5078.9  579.35  5108.9  586.06
  5118.9  587.97  5128.9  590.89  5148.9  594.07  5168.9  598.05
#Mann= 3 , 1 , 0
 4718.50    0.11       0  4990.4   0.045       0  5009.6    0.14       0
Bank Sta=4990.40,5009.60
Exp/Cntr=0.3,0.1

Type RM Length L Ch R = 1 ,23748.9,748.9,748.9,748.9
XS GIS Cut Line= 3
 1948147.1136499 843020.74043149 1948306.8435317 842594.06472003
 1948401.8241312 842362.80760810
BEGIN DESCRIPTION:
Sevenmile Creek 47.0
END DESCRIPTION:
#Sta/Elev= 28
  4554.7  592.12  4564.7  591.58  4584.7  591.03  4594.7   590.4  4634.7  589.94
  4694.7  590.71  4814.7  588.99  4914.7  583.59  4934.7  581.33  4944.7  580.49
  4954.7  579.11  4964.7  577.27  4974.7  576.36  4990.4  574.28  4991.9  571.28
  5008.1  571.28  5009.6  574.28  5010.3   577.3  5020.3  578.11  5030.3  577.76
  5040.3  577.98  5060.3  578.96  5130.3  580.47  5160.3  583.37  5210.3  589.61
  5220.3  591.22  5230.3  592.45  5260.3  595.36
#Mann= 3 , 1 , 0
 4554.70    0.11       0  4990.4   0.045       0  5009.6    0.14       0
Bank Sta=4990.40,5009.60
Exp/Cntr=0.3,0.1

Type RM Length L Ch R = 1 ,23000.0,471.3,471.3,471.3
XS GIS Cut Line= 3
  1948943.011153 842929.50684973 1948939.1988169 842790.99197147
 1948934.9131239 842520.99331444
BEGIN DESCRIPTION:
Sevenmile Creek 46.0
END DESCRIPTION:
#Sta/Elev= 22
  4855.9  597.95  4895.9  587.28  4905.9  584.14  4925.9  578.46  4935.9  575.97
  4945.9  576.23  4975.9  573.62  4985.9  574.17  4990.4  573.29  4991.9  570.29
  5008.1  570.29  5009.6  573.29  5014.5  578.08  5034.5  579.74  5044.5  580.29
  5054.5  580.21  5064.5  580.57  5074.5  581.53  5094.5  582.67  5104.5   583.5
  5144.5   588.3  5264.5   596.2
#Mann= 3 , 1 , 0
 4855.90    0.14       0  4990.4   0.045       0  5009.6    0.11       0
Bank Sta=4990.40,5009.60
Exp/Cntr=0.3,0.1

Type RM Length L Ch R = 1 ,22528.7,849.3,849.3,849.3
XS GIS Cut Line= 3
 1949490.4027254 842837.40359640 1949305.6681238 842631.39884478
 1949126.1771395 842417.71910146
BEGIN DESCRIPTION:
Sevenmile Creek 45.0
END DESCRIPTION:
#Sta/Elev= 28
  4721.1  590.81  4741.1  590.02  4751.1  589.98  4761.1  590.22  4771.1  589.39
  4781.1  587.91  4791.1  588.09  4841.1  584.02  4851.1   584.2  4871.1  582.82
  4891.1  582.45  4911.1  581.17  4931.1  579.19  4941.1  577.91  4951.1  576.33
  4961.1  575.13  4971.1  574.47  4981.1  574.15  4990.3  572.53  4991.8  569.53
  5008.1  569.53  5009.6  572.53  5097.8  578.07  5107.8  578.31  5127.8  580.15
  5197.8  584.14  5217.8  584.71  5276.8  588.91
#Mann= 3 , 1 , 0
 4721.10    0.14       0  4990.3   0.045       0  5009.6    0.11       0
Bank Sta=4990.30,5009.60
Exp/Cntr=0.3,0.1

Type RM Length L Ch R = 1 ,21679.4,543.75,543.75,543.75
XS GIS Cut Line= 3
 1949634.7349286 842776.70107024 1949771.4899643 842558.74773205
 1949801.7082956 842401.61240934
BEGIN DESCRIPTION:
Sevenmile Creek 43.0
END DESCRIPTION:
#Sta/Elev= 30
  4740.7  583.01  4750.7  582.32  4760.7  580.97  4800.7   577.2  4810.7  576.92
  4820.7  577.35  4830.7  576.09  4840.7  573.99  4860.7  572.89  4870.7  571.33
  4880.7  568.67  4890.7   566.9  4900.7  567.44  4920.7  570.35  4930.7  570.59
  4940.7  570.02  4970.7     570  4980.7  570.66  4990.4  568.63  4991.9  565.63
  5008.1  565.63  5009.6  568.63    5028  571.86    5038  573.03    5078  574.62
    5098  574.68    5118  577.03    5128  581.15    5138  582.42    5158  583.91
#Mann= 3 , 1 , 0
 4740.70    0.14       0  4990.4   0.045       0  5009.6    0.11       0
Bank Sta=4990.40,5009.60
Exp/Cntr=0.5,0.3

Type RM Length L Ch R = 1 ,21135.7,45.5,45.5,45.5
XS GIS Cut Line= 3
 1950208.9864722 843143.80080753 1950112.7367389 842904.15861439
 1950010.6916133 842598.02323782
BEGIN DESCRIPTION:
Upstream Section of Bridge/Culvert/Weir
END DESCRIPTION:
#Sta/Elev= 30
    4743  589.05    4773  585.78    4783  585.15    4793  583.07    4833   577.8
    4853   577.5    4863  576.96    4893  573.84    4913  572.66    4923  570.87
    4933  570.21    4943  567.64    4953  566.36    4963  566.77  4972.5  564.03
    4976  561.03    5024  561.03  5027.5  564.03  5037.2   574.8  5057.2  575.36
  5077.2  576.88  5117.2  578.87  5147.2  579.48  5167.2  580.39  5177.2  580.21
  5187.2  581.11  5277.2  585.12  5287.2  584.84  5307.2  585.92  5324.5  586.17
#Mann= 3 , 1 , 0
 4743.00    0.11       0  4972.5   0.045       0  5027.5    0.11       0
#XS Ineff= 2 , 0
       0 4944.85  577.88 5055.05       0  579.21
Bank Sta=4972.50,5027.50
Exp/Cntr=0.5,0.3

Type RM Length L Ch R = 3 ,21112.9,,,
BEGIN DESCRIPTION:
Mt Willing Road-TOR
Structure ID: Mt Willing Road (SC)-Bridge
Approximate Survey Structure
END DESCRIPTION:
Bridge Culvert--1,0,-1,-1, 0
Deck Dist Width WeirC Skew NumUp NumDn MinLoCord MaxHiCord MaxSubmerge Is_Ogee
10,25.5,2.6,,52,52,,,0.95,0,1,1,,
    4743  4743.6  4763.6    4773  4773.6    4783    4793  4793.6    4833  4843.6
    4853    4863    4873    4893    4903    4913    4923    4933    4943    4953
 4954.91    4955  4955.8    4963  4972.5    4976    5024  5027.5  5037.2  5044.3
 5044.89    5045  5047.2  5057.2  5077.2  5117.2  5137.2  5147.2  5157.2  5167.2
  5177.2  5187.2  5191.8  5201.8  5211.8  5241.8  5268.9  5277.2  5287.2  5297.2
  5307.2  5324.5
  588.02  587.96  585.78  584.76  584.72  584.13  582.05  581.97  578.48  577.87
  577.93  577.99  578.06  578.18  578.25  578.31  578.37  578.44   578.5  578.56
  578.58  578.58  578.58  578.63  578.69  578.71  579.01  579.04   579.1  579.14
  579.15  579.15  579.16  579.23  579.35  579.61  579.73   579.8  579.86  579.92
  579.99  580.09  580.29  580.74  581.19  582.52  583.73  584.09  583.81  584.13
  584.89  585.14
  588.02  587.95  585.77  584.75  584.71  584.12  582.04  581.96  576.77  576.61
  576.47  575.93  574.68  572.81   572.4  571.63  569.84  569.18  566.61  565.33
  565.41  576.58  576.58  576.63  576.69  576.71  577.01  577.04   577.1  577.14
  577.15  574.11  574.21  574.33  575.85  577.84  578.48  578.45  579.08  579.36
  579.18  580.08  580.28  580.73  581.18  582.51  583.72  584.09  583.81  584.13
  584.89  585.14
    4743  4743.6  4763.6    4773  4773.6    4783    4793  4793.6    4833  4843.6
    4853    4863    4873    4893    4903    4913    4923    4933    4943    4953
 4954.91    4955  4955.8    4963  4972.5    4976    5024  5027.5  5037.2  5044.3
 5044.89    5045  5047.2  5057.2  5077.2  5117.2  5137.2  5147.2  5157.2  5167.2
  5177.2  5187.2  5191.8  5201.8  5211.8  5241.8  5268.9  5277.2  5287.2  5297.2
  5307.2  5324.5
  588.02  587.96  585.78  584.76  584.72  584.13  582.05  581.97  578.48  577.87
  577.93  577.99  578.06  578.18  578.25  578.31  578.37  578.44   578.5  578.56
  578.58  578.58  578.58  578.63  578.69  578.71  579.01  579.04   579.1  579.14
  579.15  579.15  579.16  579.23  579.35  579.61  579.73   579.8  579.86  579.92
  579.99  580.09  580.29  580.74  581.19  582.52  583.73  584.09  583.81  584.13
  584.89  585.14
  587.77   587.7  585.52   584.5  584.46  583.87  581.79  581.71  576.52  576.36
  576.22  575.68  574.43  572.56  572.15  571.38  569.59  568.93  566.36  565.08
  565.16  576.33  576.33  576.38  576.44  576.46  576.76  576.79  576.85  576.89
   576.9  573.86  573.96  574.08   575.6  577.59  578.23   578.2  578.83  579.11
  578.93  579.83  580.03  580.48  580.93  582.26  583.47  583.84  583.56  583.88
  584.64  584.89
Pier Skew, UpSta & Num, DnSta & Num=,4966.9, 2 ,4966.9, 2 , 0 , 0 , 0 ,,
       1       1
  563.47  577.66
       1       1
  563.22  577.41
Pier Skew, UpSta & Num, DnSta & Num=,4989.0, 2 ,4989.0, 2 , 0 , 0 , 0 ,,
       1       1
     559  577.79
       1       1
  558.75  577.54
Pier Skew, UpSta & Num, DnSta & Num=,5011.1, 2 ,5011.1, 2 , 0 , 0 , 0 ,,
       1       1
     559  577.93
       1       1
  558.75  577.68
Pier Skew, UpSta & Num, DnSta & Num=,5033.2, 2 ,5033.2, 2 , 0 , 0 , 0 ,,
       1       1
  567.77  578.08
       1       1
  567.52  577.83
Abutment Skew #Up #Dn=, 2 , 2
 4954.80 4955.80
  576.58  565.44
 4954.80 4955.80
  576.33  565.19
BR Coef= 1 , 1 , 0 ,1.25, 0 ,,,0.8,0,2,0,
Wspro=,,,, 1 ,,,, 0 ,,,, 0 ,,,,-1 ,-1 ,-1 , 0 , 0 , 0 , 0 , 0
BC Design=,, 0 ,, 0 ,,,,,,
BR U #Sta/Elev= 52
    4743  588.02  4743.6  587.95  4763.6  585.77    4773  584.75  4773.6  584.71
    4783  584.12    4793  582.04  4793.6  581.96    4833  576.77  4843.6  576.61
    4853  576.47    4863  575.93    4873  574.68    4893  572.81    4903   572.4
    4913  571.63    4923  569.84    4933  569.18    4943  566.61    4953  565.33
 4954.91  565.41    4955  565.41  4955.8  565.44    4963  565.74  4972.5     563
    4976     560    5024     560  5027.5     563  5037.2  573.77  5044.3  574.08
 5044.89  574.11    5045  574.11  5047.2  574.21  5057.2  574.33  5077.2  575.85
  5117.2  577.84  5137.2  578.48  5147.2  578.45  5157.2  579.08  5167.2  579.36
  5177.2  579.18  5187.2  580.08  5191.8  580.28  5201.8  580.73  5211.8  581.18
  5241.8  582.51  5268.9  583.72  5277.2  584.09  5287.2  583.81  5297.2  584.13
  5307.2  584.89  5324.5  585.14
BR U #Mann= 3
 4743.00    0.11  4972.5   0.045  5027.5    0.11
BR U Banks=4972.50,5027.50
BR D #Sta/Elev= 52
    4743  587.77  4743.6   587.7  4763.6  585.52    4773   584.5  4773.6  584.46
    4783  583.87    4793  581.79  4793.6  581.71    4833  576.52  4843.6  576.36
    4853  576.22    4863  575.68    4873  574.43    4893  572.56    4903  572.15
    4913  571.38    4923  569.59    4933  568.93    4943  566.36    4953  565.08
 4954.91  565.16    4955  565.16  4955.8  565.19    4963  565.49  4972.5  562.75
    4976  559.75    5024  559.75  5027.5  562.75  5037.2  573.52  5044.3  573.83
 5044.89  573.86    5045  573.86  5047.2  573.96  5057.2  574.08  5077.2   575.6
  5117.2  577.59  5137.2  578.23  5147.2   578.2  5157.2  578.83  5167.2  579.11
  5177.2  578.93  5187.2  579.83  5191.8  580.03  5201.8  580.48  5211.8  580.93
  5241.8  582.26  5268.9  583.47  5277.2  583.84  5287.2  583.56  5297.2  583.88
  5307.2  584.64  5324.5  584.89
BR D #Mann= 3
 4743.00    0.11  4972.5   0.045  5027.5    0.11
BR D Banks=4972.50,5027.50

Type RM Length L Ch R = 1 ,21090.2,389.15,389.15,389.15
XS GIS Cut Line= 3
 1950254.3122707 843147.77849316 1950158.0625374 842908.13630002
 1950056.0174119 842602.00092346
BEGIN DESCRIPTION:
Downstream Section of Bridge/Culvert/Weir
END DESCRIPTION:
#Sta/Elev= 30
    4743  587.65    4773  584.38    4783  583.75    4793  581.67    4833   576.4
    4853   576.1    4863  575.56    4893  572.44    4913  571.26    4923  569.47
    4933  568.81    4943  566.24    4953  564.96    4963  565.37  4972.5  562.63
    4976  559.63    5024  559.63  5027.5  562.63  5037.2   573.4  5057.2  573.96
  5077.2  575.48  5117.2  577.47  5147.2  578.08  5167.2  578.99  5177.2  578.81
  5187.2  579.71  5277.2  583.72  5287.2  583.44  5307.2  584.52  5324.5  584.77
#Mann= 3 , 1 , 0
 4743.00    0.11       0  4972.5   0.045       0  5027.5    0.11       0
#XS Ineff= 2 , 0
       0 4944.85  577.88 5055.05       0  579.21
Bank Sta=4972.50,5027.50
Exp/Cntr=0.5,0.3

Type RM Length L Ch R = 1 ,20701.0,702.1,702.1,702.1
XS GIS Cut Line= 3
 1950620.9380182 843090.95244130 1950553.5578248 842956.19205463
 1950459.4183393 842791.11505693
BEGIN DESCRIPTION:
Sevenmile Creek 41.0
END DESCRIPTION:
#Sta/Elev= 20
  4832.8   579.5  4882.8  572.04  4902.8  568.04  4912.8  565.58  4962.8  558.62
  4972.8  558.56  4983.5  558.93  4990.4  558.41  4991.9  555.41  5008.1  555.41
  5009.6  558.41  5013.5  562.36  5023.5  563.99  5033.5  564.66  5063.5  564.96
  5083.5  564.56  5093.5  565.37  5133.5  573.62  5153.5  576.64  5173.5  580.01
#Mann= 3 , 1 , 0
 4832.80    0.11       0  4990.4   0.045       0  5009.6    0.11       0
Bank Sta=4990.40,5009.60
Exp/Cntr=0.3,0.1

Type RM Length L Ch R = 1 ,19998.9,591.2,591.2,591.2
XS GIS Cut Line= 3
 1950999.0860566 842995.55639702 1950905.0250064 842630.36517266
 1950856.3892196 842543.00088893
BEGIN DESCRIPTION:
Sevenmile Creek 40.0
END DESCRIPTION:
#Sta/Elev= 30
  4624.9  573.36  4644.9  568.91  4654.9  566.96  4674.9  564.27  4684.9  563.28
  4704.9   562.4  4714.9  562.53  4724.9  562.11  4784.9   562.4  4794.9  562.12
  4804.9  562.49  4814.9  562.14  4854.9  562.86  4904.9  562.03  4924.9  560.85
  4944.9   558.9  4954.9  559.08  4964.9  558.84  4974.9     557  4984.9  556.09
  4990.3  555.31  4991.8  552.31  5008.1  552.31  5009.6  555.31    5012  559.74
    5042   560.8    5052  563.26    5062  565.11    5072  567.32    5102  575.54
#Mann= 3 , 1 , 0
 4624.90    0.11       0  4990.3   0.045       0  5009.6    0.11       0
Bank Sta=4990.30,5009.60
Exp/Cntr=0.3,0.1

Type RM Length L Ch R = 1 ,19407.7,538.2,538.2,538.2
XS GIS Cut Line= 3
 1951310.4334127 843005.70043344 1951362.5075860 842430.51751947
 1951370.9273633 842350.99740039
BEGIN DESCRIPTION:
Sevenmile Creek 39.0
END DESCRIPTION:
#Sta/Elev= 30
  4420.8  574.04  4450.8  566.71  4460.8  564.79  4490.8  560.54  4540.8  560.64
  4570.8  561.35  4620.8  559.48  4740.8  558.77  4760.8  558.14  4780.8  558.48
  4790.8  557.99  4810.8  559.33  4820.8  557.76  4830.8  557.65  4850.8  557.89
  4880.8   559.4  4900.8  558.74  4930.8  559.11  4970.8  555.23  4990.3  554.35
  4991.8  551.35  5008.1  551.35  5009.6  554.35  5018.3  555.45  5028.3  555.19
  5038.3  553.63  5048.3  554.28  5058.3  565.21  5068.3  572.41  5078.3  575.32
#Mann= 3 , 1 , 0
 4420.80    0.14       0  4990.3   0.045       0  5009.6    0.14       0
Bank Sta=4990.30,5009.60
Exp/Cntr=0.3,0.1

Type RM Length L Ch R = 1 ,18869.5,433,433,433
XS GIS Cut Line= 3
 1951828.7230625 842797.43978816 1951853.6994083 842601.47153605
 1951862.4853764 842511.85466126
BEGIN DESCRIPTION:
Sevenmile Creek 38.0
END DESCRIPTION:
#Sta/Elev= 23
  4801.4  570.19  4831.4  567.05  4871.4  561.64  4881.4  560.56  4891.4  559.83
  4911.4  556.64  4921.4  555.86  4931.4  555.58  4941.4  555.92  4961.4  555.79
  4971.4  556.12  4981.4  556.97  4989.8  551.96  4991.3  548.96  5008.7  548.96
  5010.2  551.96    5019  555.57    5029  555.69    5039  556.16    5049  558.93
    5069  565.05    5079  568.75    5089  575.09
#Mann= 3 , 1 , 0
 4801.40    0.14       0  4989.8   0.045       0  5010.2    0.14       0
Bank Sta=4989.80,5010.20
Exp/Cntr=0.3,0.1

Type RM Length L Ch R = 1 ,18436.5,370.1,370.1,370.1
XS GIS Cut Line= 3
 1951967.8387665 842889.54983386 1952039.1002432  842851.8830533
 1952144.9507172 842795.36095555
BEGIN DESCRIPTION:
Sevenmile Creek 37.0
END DESCRIPTION:
#Sta/Elev= 17
  4917.9  569.76  4937.9  565.32  4957.9  558.41  4977.9  554.02  4987.9  551.09
  4989.8  550.02  4991.3  547.02  5008.8  547.02  5010.3  550.02  5018.5   550.2
  5038.5  552.29  5058.5  553.36  5068.5  554.83  5078.5   556.8  5098.5  563.44
  5108.5  566.44  5118.5  569.11
#Mann= 3 , 1 , 0
 4917.90    0.14       0  4989.8   0.045       0  5010.3    0.14       0
Bank Sta=4989.80,5010.30
Exp/Cntr=0.3,0.1

Type RM Length L Ch R = 1 ,18066.4,460.1,460.1,460.1
XS GIS Cut Line= 3
 1952028.1167912 843231.02481255 1952084.8485012 843198.60669257
 1952408.0314062 843040.10297482
BEGIN DESCRIPTION:
Sevenmile Creek 36.0
END DESCRIPTION:
#Sta/Elev= 25
  4936.2  571.76  4956.2  561.99  4989.7  548.36  4991.2  545.36  5008.7  545.36
  5010.2  548.36  5011.5  553.03  5021.5  553.48  5041.5  553.06  5051.5  553.58
  5071.5  553.91  5081.5  553.54  5091.5   552.9  5111.5  552.87  5131.5  555.42
  5181.5  559.12  5191.5  559.41  5201.5  559.16  5221.5  557.05  5231.5  556.97
  5241.5  557.74  5271.5  559.09  5291.5  561.14  5321.5  566.94  5361.5   572.8
#Mann= 3 , 1 , 0
 4936.20    0.14       0  4989.7   0.045       0  5010.2    0.14       0
Bank Sta=4989.70,5010.20
Exp/Cntr=0.3,0.1

Type RM Length L Ch R = 1 ,17606.3,606.3,606.3,606.3
XS GIS Cut Line= 3
 1952378.5799454 843557.72080186 1952424.3487313 843499.58207388
 1952555.6329004 843240.99204374
BEGIN DESCRIPTION:
Sevenmile Creek 35.0
END DESCRIPTION:
#Sta/Elev= 28
  4924.7  567.91  4934.7   564.4  4954.7   556.1  4964.7  552.65  4974.7  551.59
  4989.8   546.3  4991.3   543.3  5008.7   543.3  5010.2   546.3  5018.7  550.21
  5058.7  553.26  5078.7  553.56  5088.7  552.72  5118.7  553.26  5128.7  552.84
  5138.7  552.01  5148.7  551.75  5158.7  551.85  5168.7  551.55  5178.7  551.69
  5198.7  552.61  5218.7  552.46  5238.7  553.59  5248.7  555.42  5258.7  556.42
  5268.7  558.55  5278.7  561.82  5288.7  565.76
#Mann= 3 , 1 , 0
 4924.70    0.14       0  4989.8   0.045       0  5010.2    0.14       0
Bank Sta=4989.80,5010.20
Exp/Cntr=0.3,0.1

Type RM Length L Ch R = 1 ,17000.0,289.8,289.8,289.8
XS GIS Cut Line= 3
 1952962.7916968 843357.64074422 1952895.9824257 843301.28961018
 1952759.9730414 843183.38668690
BEGIN DESCRIPTION:
Sevenmile Creek 34.0
END DESCRIPTION:
#Sta/Elev= 21
  4912.6  565.23  4932.6  559.89  4942.6   556.6  4952.6   553.6  4962.6  551.06
  4972.6  548.84  4982.6  546.14  4989.8  543.85  4991.3  540.85  5008.7  540.85
  5010.2  543.85    5040  547.94    5050  547.83    5060  547.31    5080   549.4
    5090  550.72    5110  552.26    5140  556.27    5150  558.41    5170  561.89
    5180   563.9
#Mann= 3 , 1 , 0
 4912.60    0.14       0  4989.8   0.045       0  5010.2    0.14       0
Bank Sta=4989.80,5010.20
Exp/Cntr=0.3,0.1

Type RM Length L Ch R = 1 ,16710.2,325.7,325.7,325.7
XS GIS Cut Line= 3
 1953095.2792476 843196.52120889 1952978.1434329 843022.83706989
 1952803.0414962 842926.18080083
BEGIN DESCRIPTION:
Sevenmile Creek 33.0
END DESCRIPTION:
#Sta/Elev= 18
  4798.3  561.65  4808.3  560.81  4848.3  558.86  4928.3  552.75  4938.3  551.54
  4948.3  549.21  4958.3  547.44  4989.8  542.87  4991.3  539.87  5008.7  539.87
  5010.2  542.87  5017.8  545.51  5037.8   548.2  5047.8  548.54  5107.8  549.59
  5127.8  551.68  5137.8  552.98  5207.8   563.7
#Mann= 3 , 1 , 0
 4798.30    0.14       0  4989.8   0.045       0  5010.2    0.14       0
Bank Sta=4989.80,5010.20
Exp/Cntr=0.3,0.1

Type RM Length L Ch R = 1 ,16384.5,765.7,765.7,765.7
XS GIS Cut Line= 3
 1953365.7925353 843125.95130598 1953050.3775244 842719.45388553
 1952928.7371943 842536.16023746
BEGIN DESCRIPTION:
Sevenmile Creek 32.0
END DESCRIPTION:
#Sta/Elev= 30
  4479.9  560.72  4489.9  559.11  4539.9  553.97  4559.9  551.06  4579.9  549.91
  4589.9  548.57  4599.9  548.35  4619.9   548.8  4629.9  548.05  4639.9  548.11
  4659.9  547.19  4839.9  547.84  4889.9  544.66  4899.9  544.98  4909.9  546.37
  4929.9  547.45  4959.9  547.47  4989.8  541.76  4991.3  538.76  5008.7  538.76
  5010.2  541.76  5014.4  546.28  5024.4  547.71  5034.4  548.37  5074.4  548.66
  5094.4  547.96  5154.4  547.18  5174.4  548.75  5184.4  551.11  5214.4  563.25
#Mann= 3 , 1 , 0
 4479.90    0.14       0  4989.8   0.045       0  5010.2    0.14       0
Bank Sta=4989.80,5010.20
Exp/Cntr=0.3,0.1

Type RM Length L Ch R = 1 ,15618.8,731.7,731.7,731.7
XS GIS Cut Line= 3
 1953685.4859995 842926.06533934 1953584.9098016  842842.2518411
 1953124.0457911 842506.87060573
BEGIN DESCRIPTION:
Sevenmile Creek 31.0
END DESCRIPTION:
#Sta/Elev= 30
  4865.8  559.37  4885.8  553.02  4895.8  550.76  4915.8  547.99  4925.8  547.28
  4955.8  547.33  4975.8  544.64  4985.8  542.48  4989.8  539.59  4991.3  536.59
  5008.7  536.59  5010.2  539.59  5016.7  544.44  5056.7  544.84  5126.7  544.81
  5146.7  544.04  5166.7  543.94  5196.7  545.22  5206.7  545.24  5236.7  544.18
  5256.7  545.29  5276.7  545.53  5366.7  544.81  5376.7  545.16  5426.7  544.55
  5446.7  545.37  5466.7  548.49  5516.7  552.44  5526.7  554.28  5566.7  560.06
#Mann= 3 , 1 , 0
 4865.80    0.14       0  4989.8   0.045       0  5010.2    0.14       0
Bank Sta=4989.80,5010.20
Exp/Cntr=0.3,0.1

Type RM Length L Ch R = 1 ,14887.1,346.8,346.8,346.8
XS GIS Cut Line= 3
 1953639.8455857 842385.19838102 1953320.0514661 842300.49615474
 1953154.1204786 842263.62260197
BEGIN DESCRIPTION:
Sevenmile Creek 30.0
END DESCRIPTION:
#Sta/Elev= 21
  4666.1  558.15  4716.1  553.49  4826.1  545.03  4836.1  544.69  4856.1  544.86
  4976.1  544.46  4986.1  543.63  4989.8  537.78  4991.3  534.78  5008.7  534.78
  5010.2  537.78  5016.9  542.84  5026.9  542.87  5036.9   542.4  5056.9  539.86
  5066.9  539.31  5076.9  539.81  5096.9     543  5106.9  546.53  5116.9  552.79
  5166.9  572.09
#Mann= 3 , 1 , 0
 4666.10    0.11       0  4989.8    0.05       0  5010.2    0.14       0
Bank Sta=4989.80,5010.20
Exp/Cntr=0.3,0.1

Type RM Length L Ch R = 1 ,14540.3,442.2,442.2,442.2
XS GIS Cut Line= 3
 1953755.2721548 842233.27070163 1953488.5976796 842021.19100088
 1953330.9661127 841882.47522198
BEGIN DESCRIPTION:
Sevenmile Creek 29.0
END DESCRIPTION:
#Sta/Elev= 30
  4658.9  564.19  4708.9   555.4  4738.9  551.49  4758.9  549.48  4768.9  548.97
  4778.9  548.86  4798.9  546.96  4808.9  546.59  4858.9   546.9  4878.9  547.89
  4918.9  547.47  4958.9  544.28  4968.9  543.14  4978.9  542.57  4988.9  540.97
  4989.8  537.12  4991.3  534.12  5008.7  534.12  5010.2  537.12  5019.6  540.85
  5029.6  541.94  5079.6  541.82  5099.6  543.93  5109.6  543.75  5119.6  544.51
  5139.6  547.22  5149.6  548.11  5159.6  549.59  5169.6  552.55  5209.6  567.01
#Mann= 3 , 1 , 0
 4658.90    0.11       0  4989.8    0.05       0  5010.2    0.14       0
Bank Sta=4989.80,5010.20
Exp/Cntr=0.3,0.1

Type RM Length L Ch R = 1 ,14098.1,672.9,672.9,672.9
XS GIS Cut Line= 3
 1953837.4101068 842118.90237829 1953753.4560151 841729.84683178
 1953722.4191546 841634.79644621
BEGIN DESCRIPTION:
Sevenmile Creek 28.0
END DESCRIPTION:
#Sta/Elev= 30
  4602.4  558.12  4642.4  551.39  4662.4  548.73  4702.4  546.38  4712.4  546.28
  4722.4  546.65  4742.4  545.95  4762.4  546.42  4792.4   544.7  4802.4  543.75
  4822.4   540.5  4832.4  539.73  4842.4   539.3  4862.4  540.86  4882.4  541.13
  4912.4  541.22  4922.4  541.61  4932.4  541.19  4952.4  541.88  4962.4  541.15
  4972.4  540.69  4982.4  539.67  4989.8  535.63  4991.3  532.63  5008.7  532.63
  5010.2  535.63  5020.4  538.19  5040.4  546.65  5050.4  549.89  5100.4  566.89
#Mann= 3 , 1 , 0
 4602.40    0.11       0  4989.8    0.05       0  5010.2    0.14       0
Bank Sta=4989.80,5010.20
Exp/Cntr=0.3,0.1

Type RM Length L Ch R = 1 ,13425.2,476.2,476.2,476.2
XS GIS Cut Line= 3
 1954400.6885993 841875.74280953 1954331.3287473 841761.14827143
 1954262.0898513 841651.18061309
BEGIN DESCRIPTION:
Sevenmile Creek 27.0
END DESCRIPTION:
#Sta/Elev= 18
  4864.4  560.88  4894.4  550.87  4914.4  544.79  4924.4  540.88  4934.4  538.54
  4974.4   532.9  4984.4     534  4989.7  531.62  4991.2  528.62  5008.7  528.62
  5010.2  531.62  5038.3  539.06  5048.3  538.48  5058.3  538.45  5068.3  541.28
  5078.3  544.52  5098.3  551.94  5128.3  555.96
#Mann= 3 , 1 , 0
 4864.40    0.11       0  4989.7    0.05       0  5010.2    0.14       0
Bank Sta=4989.70,5010.20
Exp/Cntr=0.3,0.1

Type RM Length L Ch R = 1 ,12949.0,359.3,359.3,359.3
XS GIS Cut Line= 3
 1954639.4200676 841515.67228067 1954581.7402645 841493.88213283
 1954307.2507168 841496.28993588
BEGIN DESCRIPTION:
Sevenmile Creek 26.0
END DESCRIPTION:
#Sta/Elev= 25
  4932.4  552.49  4942.4  549.22  4952.4  544.89  4962.4  539.96  4972.4  536.11
  4982.4  533.95  4989.8  530.29  4991.3  527.29  5008.7  527.29  5010.2  530.29
  5014.1  532.77  5024.1  535.18  5034.1  537.33  5044.1  538.23  5054.1  538.52
  5074.1  538.52  5104.1  539.88  5124.1  540.26  5154.1  541.89  5174.1   542.3
  5194.1  543.73  5204.1  544.85  5214.1  545.49  5244.1  547.68  5268.6  551.16
#Mann= 3 , 1 , 0
 4932.40    0.11       0  4989.8    0.05       0  5010.2    0.14       0
Bank Sta=4989.80,5010.20
Exp/Cntr=0.3,0.1

Type RM Length L Ch R = 1 ,12589.7,665.4,665.4,665.4
XS GIS Cut Line= 3
 1954721.7385782 841198.65108233 1954644.3431438 841144.75069051
 1954333.7365503 841099.00243255
BEGIN DESCRIPTION:
Sevenmile Creek 25.0
END DESCRIPTION:
#Sta/Elev= 29
  4898.6   554.7  4918.6  549.67  4928.6  547.66  4938.6   545.3  4958.6   539.7
  4968.6  536.21  4978.6  533.67  4989.8  530.27  4991.3  527.27  5008.7  527.27
  5010.2  530.27  5012.9  534.62  5032.9   536.6  5042.9  537.21  5052.9  537.52
  5072.9  536.74  5082.9  536.87  5092.9  536.54  5112.9   536.7  5132.9  535.97
  5152.9  536.22  5162.9  536.01  5172.9  536.67  5212.9  539.77  5242.9  541.33
  5252.9  542.13  5272.9   544.4  5292.9  545.05  5306.9  545.87
#Mann= 3 , 1 , 0
 4898.60    0.11       0  4989.8    0.05       0  5010.2    0.14       0
Bank Sta=4989.80,5010.20
Exp/Cntr=0.3,0.1

Type RM Length L Ch R = 1 ,11924.3,514.2,514.2,514.2
XS GIS Cut Line= 3
 1954795.1501826 841007.17116068 1954759.9176903  840610.2184133
 1954740.5616497 840575.22864772
BEGIN DESCRIPTION:
Sevenmile Creek 24.0
END DESCRIPTION:
#Sta/Elev= 28
  4600.4  550.78  4610.4  549.25  4620.4  549.51  4630.4  549.38  4640.4  547.85
  4650.4  547.76  4660.4  546.98  4670.4  547.03  4680.4  546.61  4700.4  545.26
  4740.4  539.56  4770.4  536.54  4780.4  536.68  4820.4   536.1  4830.4  536.29
  4840.4  536.03  4880.4  536.95  4900.4   536.7  4910.4  536.01  4940.4  532.21
  4950.4  530.53  4980.4  532.51  4989.8  530.22  4991.3  527.22  5008.7  527.22
  5010.2  530.22  5018.9  545.56  5038.9  560.14
#Mann= 3 , 1 , 0
 4600.40    0.11       0  4989.8    0.05       0  5010.2    0.14       0
Bank Sta=4989.80,5010.20
Exp/Cntr=0.3,0.1

Type RM Length L Ch R = 1 ,11410.1,444.1,444.1,444.1
XS GIS Cut Line= 3
         1954825          841075 1954976.6199648 840976.20447697
 1955081.1711069 840917.22690960
BEGIN DESCRIPTION:
Sevenmile Creek 23.0
END DESCRIPTION:
#Sta/Elev= 19
  4822.5  550.33  4842.5  546.48  4862.5   543.9  4882.5  540.39  4922.5   535.2
  4952.5  530.33  4982.5  527.78  4987.3  525.45  4988.8  522.45  5011.2  522.45
  5012.7  525.45  5023.5  530.35  5033.5  531.57  5043.5  533.53  5053.5  535.06
  5063.5   537.2  5073.5  539.95  5103.5  547.02  5123.5  550.59
#Mann= 3 , 1 , 0
 4822.50    0.11       0  4987.3    0.05       0  5012.7    0.14       0
Bank Sta=4987.30,5012.70
Exp/Cntr=0.3,0.1
