--- S_Fork_Little_River_FINAL.prj (project) ---

Proj Title=South Fork Little River
Current Plan=p01
Default Exp/Contr=0.3,0.1
English Units
Geom File=g01
Flow File=f01
Plan File=p01
Y Axis Title=Elevation
X Axis Title(PF)=Main Channel Distance
X Axis Title(XS)=Station
BEGIN DESCRIPTION:
####(Watershed Name)####
SOUTH FORK LITTLE RIVER
HCFCD Unit X###-##-##
(Flood Hazard, Floodway) Model
10, 2, 1, 0.2% Event
Filename:  N:\NC_flood\60138\Orange\URS\Limited_Detail\ENG\South Fork Little River\South Fork Little River.prj
Prepared by:  ________     Date: ________
Reviewed by:  ________     Date: ________
STATUS (Draft RAS, SVSQ, FINAL)
END DESCRIPTION:
DSS Export Rating Curves= 0
DSS Export Rating Curve Sorted= 0
DSS Export Volume Flow Curves= 0
DXF OffsetX= 0
DXF OffsetY= 0
DXF ScaleX= 1
DXF ScaleY= 10

--- S_Fork_Little_River_FINAL.p01 (plan) ---

Plan Title=100 Year Single
Version=Version 3.0.1  Mar 2001
Short Identifier=100 Year Sin
Geom File=g01
Flow File=f01
Subcritical Flow
K Sum by GR= 0
Std Step Tol= 0.01
Critical Tol= 0.01
Num of Std Step Trials= 20
Max Error Tol= 0.3
Flow Tol Ratio= 0.001
Split Flow NTrial= 30
Split Flow Tol= 0.02
Split Flow Ratio= 0.02
Log Output Level= 0
Friction Slope Method= 1
Unsteady Friction Slope Method= 2
Parabolic Critical Depth
Global Vel Dist= 0 , 0 , 0
Global Log Level= 0
CheckData=True
Encroach Param=-1 ,0,0, 2
Encroach River=South Fork Littl
Encroach Reach=Reach - 1
Encroach Node=89759.9
       1 4979.69  5041.1
Encroach Node=89691.2
       1    4969    5023
Encroach Node=89670.9
       1    4969    5023
Encroach Node=89650.7
       1    4969    5023
Encroach Node=89106.6
       1 4878.95 5023.78
Encroach Node=88500.0
       1 4853.37 5048.69
Encroach Node=88000.0
       1 4899.27 5054.49
Encroach Node=87500.0
       1 4855.28 5015.17
Encroach Node=87154.7
       1 4957.88 5068.26
Encroach Node=86553.7
       1    4995 5058.48
Encroach Node=86000.0
       1    4970    5025
Encroach Node=85568.2
       1 4961.95 5028.14
Encroach Node=85041.4
       1    4950    5045
Encroach Node=84552.0
       1 4990.41 5015.81
Encroach Node=84104.9
       1 4984.18 5026.93
Encroach Node=83500.0
       1 4942.05 5011.01
Encroach Node=83112.0
       1 4970.78 5184.47
Encroach Node=82500.0
       1  4817.3 5031.83
Encroach Node=81858.0
       1    4972    5027
Encroach Node=81835.0
       1    4972    5027
Encroach Node=81812.0
       1    4972    5027
Encroach Node=81500.0
       1 4815.04    5008
Encroach Node=81000.0
       1 4914.81  5087.1
Encroach Node=80302.6
       1 4899.16 5038.43
Encroach Node=79449.3
       1  4838.6 5168.12
Encroach Node=79079.0
       1 4842.11 5152.97
Encroach Node=78500.0
       1 4982.26 5257.03
Encroach Node=78000.0
       1 4960.58 5131.62
Encroach Node=77500.0
       1 4935.12 5069.96
Encroach Node=77000.0
       1    4987  5262.9
Encroach Node=76473.6
       1    4969    5030
Encroach Node=76441.8
       1    4969    5030
Encroach Node=76410.1
       1    4969    5030
Encroach Node=76117.4
       1  4981.3 5390.92
Encroach Node=75500.0
       1  4770.2 5082.75
Encroach Node=75097.4
       1 4657.85 5083.51
Encroach Node=74398.8
       1 4598.78    5016
Encroach Node=74000.0
       1 4706.16    5030
Encroach Node=73433.4
       1 4766.74    5015
Encroach Node=72924.9
       1  4799.4 5173.38
Encroach Node=72408.0
       1    4820    5050
Encroach Node=71752.2
       1    4875    5050
Encroach Node=71731.9
       1    4875    5050
Encroach Node=71711.7
       1    4875    5050
Encroach Node=71319.0
       1 4936.43 5037.18
Encroach Node=70855.4
       1    4975 5067.49
Encroach Node=70500.0
       1    4981 5090.56
Encroach Node=70000.0
       1 4981.57 5088.94
Encroach Node=69369.1
       1    4970  5135.4
Encroach Node=68557.5
       1 4677.01    5030
Encroach Node=68000.0
       1  4735.5    5030
Encroach Node=67427.3
       1 4495.84    5039
Encroach Node=66668.0
       1 4748.67 5031.06
Encroach Node=66000.0
       1 4930.71    5029
Encroach Node=65393.3
       1    4966 5017.44
Encroach Node=65000.0
       1 4876.87 5031.22
Encroach Node=64371.8
       1 4912.06    5027
Encroach Node=63954.8
       1 4836.28    5027
Encroach Node=63396.4
       1 4927.25 5019.32
Encroach Node=62959.0
       1 4982.93 5023.75
Encroach Node=62446.8
       1    4965    5040
Encroach Node=62000.0
       1    4980    5030
Encroach Node=61500.0
       1 4985.78 5072.42
Encroach Node=60934.2
       1    4976    5250
Encroach Node=60500.0
       1 4942.75 5024.47
Encroach Node=60000.0
       1 4957.66 5036.28
Encroach Node=59500.0
       1 4911.25 5025.63
Encroach Node=59032.5
       1  4981.5 5087.27
Encroach Node=58500.0
       1 4954.41 5039.15
Encroach Node=58000.0
       1    4968 5036.48
Encroach Node=57379.6
       1    4976    5031
Encroach Node=56697.0
       1    4969    5030
Encroach Node=56678.7
       1    4969    5030
Encroach Node=56660.5
       1    4969    5030
Encroach Node=55965.6
       1    4983 5061.18
Encroach Node=55298.6
       1    4967 5062.02
Computation Interval=1HOUR
Output Interval=1HOUR
Run HTab= 0
Run UNet= 0
Run PostProcess= 0
UNET Theta= 1
UNET ZTol= 0.02
UNET ZSATol= 0.1
UNET MxIter= 20
UNET MaxInSteps= 20
UNET DtIC= 0
UNET DtMin= 0
UNET MaxCRTS= 20
UNET WFStab= 2
UNET SFStab= 1
UNET WFX= 1
UNET SFX= 1
UNET Convert EG Bridges=-1
UNET Use Existing IB Tables=-1
Instantaneous Interval=1HOUR
DSS File=dss
Write IC File= 0
Write Velocity= 0
Write Detailed= 0

--- S_Fork_Little_River_FINAL.f01 (steady flow) ---

Flow Title= 100 Year Single
Version=Version 3.0.1  Mar 2001
Number of Profiles= 2
Profile Names=100-Year,100 yr fw
River Rch & RM=South Fork Littl,Reach - 1       ,89759.9
    1075    1075
River Rch & RM=South Fork Littl,Reach - 1       ,89106.6
    1410    1410
River Rch & RM=South Fork Littl,Reach - 1       ,85041.4
    1688    1688
River Rch & RM=South Fork Littl,Reach - 1       ,80302.6
    2296    2296
River Rch & RM=South Fork Littl,Reach - 1       ,72924.9
    2487    2487
River Rch & RM=South Fork Littl,Reach - 1       ,71319.0
    4012    4012
River Rch & RM=South Fork Littl,Reach - 1       ,60934.2
    4159    4159
River Rch & RM=South Fork Littl,Reach - 1       ,56697.0
    4282    4282
Boundary for River Rch & Prof#=South Fork Littl,Reach - 1       , 1
Up Type= 0
Dn Type= 1
Dn Known WS=551.81
Boundary for River Rch & Prof#=South Fork Littl,Reach - 1       , 2
Up Type= 0
Dn Type= 1
Dn Known WS=552.51
DSS Import GetInterval= 0
DSS Import GetPeak= 0
DSS Import FillOption= 0

--- S_Fork_Little_River_FINAL.g01 (geometry) ---

Geom Title=Geom 01 by CodeH2 for Windows

River Reach=South Fork Littl,Reach - 1
Reach XY= 30
       1964653.5 893504.77750112      1964796.67       892810.03
      1964579.82       892312.06      1965205.81       891453.02
      1965169.24        891074.7      1967098.43       888853.94
      1968100.65        888936.5      1969050.61        888312.6
      1969397.57       888529.97      1969678.69       888129.71
      1970315.14       888097.31      1971040.94       886053.69
      1970944.79        885585.5       1972150.8       884647.03
      1972989.98       884541.48      1973768.03       884021.56
      1976525.37       880947.62      1977447.61       881071.07
      1978822.99       880402.99       1978170.8       879869.26
      1978323.93       879632.91       1978870.7       879651.21
       1980071.6       878339.63      1979633.85       877780.37
      1979911.81       877350.94      1980026.79        877786.4
      1980405.54       877900.02      1981693.31       876744.82
      1982217.89       877439.84 1982606.0015812 877195.64945346

Type RM Length L Ch R = 1 ,89759.9,68.75,68.75,68.75
XS GIS Cut Line= 3
 1964876.8244981 893522.95885348 1964654.7712075 893504.81118675
 1964460.5618473 893504.87602444
BEGIN DESCRIPTION:
South Fork Little River 179.0
END DESCRIPTION:
#Sta/Elev= 20
  4775.9  644.01  4805.9  643.58  4865.9  641.54  4915.9  638.12  4935.9  636.11
  4945.9  635.55  4965.9  636.04  4985.9  635.37  4995.9  633.72  4997.4   629.1
  4998.9   626.1    5001   626.1  5002.5   629.1  5008.7  634.65  5018.7  635.53
  5038.7  634.54  5058.7  635.59  5088.7  636.58  5158.7  640.75  5192.9  645.02
#Mann= 3 , 1 , 0
 4775.90    0.12       0  4997.4    0.04       0  5002.5    0.12       0
Bank Sta=4997.40,5002.50
Exp/Cntr=0.5,0.3

Type RM Length L Ch R = 1 ,89691.2,40.5,40.5,40.5
XS GIS Cut Line= 3
 1964933.6363307 893463.00766759 1964668.9347501 893438.54679546
 1964449.8980395 893425.13638460
BEGIN DESCRIPTION:
Upstream Section of Bridge/Culvert/Weir
END DESCRIPTION:
#Sta/Elev= 28
  4730.7  644.01  4783.1   642.9  4840.7   641.4  4860.7  640.88  4883.1   640.3
  4933.1   636.6 4978.41   629.2  4978.5  629.18    4983  628.45  4991.5  627.06
    4994  624.96    5006  624.96  5008.5  627.06    5017  630.52 5021.39  632.31
  5021.5  632.35  5028.4  635.16  5038.4  633.96  5048.4  635.24  5058.4  635.97
  5118.4  638.31  5128.4   638.4  5156.5  640.58  5168.4  641.51  5186.5  643.06
  5198.4  644.08  5206.5  645.19    5216  646.49
#Mann= 3 , 1 , 0
 4730.70    0.12       0  4991.5    0.04       0  5008.5    0.12       0
#XS Ineff= 2 , 0
       0  4968.3   640.9  5031.6       0   641.3
Bank Sta=4991.50,5008.50
Exp/Cntr=0.5,0.3

Type RM Length L Ch R = 3 ,89670.9,,,
BEGIN DESCRIPTION:
Hawkins Road-TOR
Structure ID: Hawkins Road (SFLR)-Bridge
Approximate Survey Structure
END DESCRIPTION:
Bridge Culvert--1,0,-1,-1, 0
Deck Dist Width WeirC Skew NumUp NumDn MinLoCord MaxHiCord MaxSubmerge Is_Ogee
10,20.5,2.6,,28,28,,,0.95,0,1,1,,
  4730.7  4783.1  4840.7  4860.7  4883.1  4933.1 4978.41  4978.5    4983  4991.5
    4994    5006  5008.5    5017 5021.39  5021.5  5028.4  5038.4  5048.4  5058.4
  5118.4  5128.4  5156.5  5168.4  5186.5  5198.4  5206.5    5216
  643.85  642.75  641.25   640.9  640.96  641.08  641.19  641.19   641.2  641.22
  641.23  641.26  641.26  641.29   641.3   641.3  641.31  641.34  641.36  641.39
  641.54  641.56  641.63  642.38  643.51  643.93  645.04  646.33
  643.85  642.74  641.24  640.72  640.14  636.44  629.04  639.59   639.6  639.62
  639.63  639.66  639.66  639.69   639.7  632.19     635   633.8  635.08  635.81
  638.15  638.24  640.42  641.35   642.9  643.92  645.03  646.33
  4730.7  4783.1  4840.7  4860.7  4883.1  4933.1 4978.41  4978.5    4983  4991.5
    4994    5006  5008.5    5017 5021.39  5021.5  5028.4  5038.4  5048.4  5058.4
  5118.4  5128.4  5156.5  5168.4  5186.5  5198.4  5206.5    5216
  643.85  642.75  641.25   640.9  640.96  641.08  641.19  641.19   641.2  641.22
  641.23  641.26  641.26  641.29   641.3   641.3  641.31  641.34  641.36  641.39
  641.54  641.56  641.63  642.38  643.51  643.93  645.04  646.33
   643.6  642.49  640.99  640.47  639.89  636.19  628.79  639.34  639.35  639.37
  639.38  639.41  639.41  639.44  639.45  631.94  634.75  633.55  634.83  635.56
   637.9  637.99  640.17   641.1  642.65  643.67  644.78  646.08
Pier Skew, UpSta & Num, DnSta & Num=,4988.6, 2 ,4988.6, 2 , 0 , 0 , 0 ,,
       1       1
  626.29  640.61
       1       1
  626.04  640.36
Pier Skew, UpSta & Num, DnSta & Num=,5000.0, 2 ,5000.0, 2 , 0 , 0 , 0 ,,
       1       1
   623.8  640.65
       1       1
  623.55   640.4
Pier Skew, UpSta & Num, DnSta & Num=,5011.3, 2 ,5011.3, 2 , 0 , 0 , 0 ,,
       1       1
  626.84  640.67
       1       1
  626.59  640.42
Abutment Skew #Up #Dn=, 2 , 2
 4978.30 4983.00
  639.59  628.29
 4978.30 4983.00
  639.34  628.04
Abutment Skew #Up #Dn=, 2 , 2
 5017.00 5021.59
  630.36  639.70
 5017.00 5021.59
  630.11  639.45
BR Coef= 1 , 1 , 0 ,1.25, 0 ,,,0.8,0,2,0,
Wspro=,,,, 1 ,,,, 0 ,,,, 0 ,,,,-1 ,-1 ,-1 , 0 , 0 , 0 , 0 , 0
BC Design=,, 0 ,, 0 ,,,,,,
BR U #Sta/Elev= 28
  4730.7  643.85  4783.1  642.74  4840.7  641.24  4860.7  640.72  4883.1  640.14
  4933.1  636.44 4978.41  629.04  4978.5  629.02    4983  628.29  4991.5   626.9
    4994   624.8    5006   624.8  5008.5   626.9    5017  630.36 5021.39  632.15
  5021.5  632.19  5028.4     635  5038.4   633.8  5048.4  635.08  5058.4  635.81
  5118.4  638.15  5128.4  638.24  5156.5  640.42  5168.4  641.35  5186.5   642.9
  5198.4  643.92  5206.5  645.03    5216  646.33
BR U #Mann= 3
 4730.70    0.12  4991.5    0.04  5008.5    0.12
BR U Banks=4991.50,5008.50
BR D #Sta/Elev= 28
  4730.7   643.6  4783.1  642.49  4840.7  640.99  4860.7  640.47  4883.1  639.89
  4933.1  636.19 4978.41  628.79  4978.5  628.77    4983  628.04  4991.5  626.65
    4994  624.55    5006  624.55  5008.5  626.65    5017  630.11 5021.39   631.9
  5021.5  631.94  5028.4  634.75  5038.4  633.55  5048.4  634.83  5058.4  635.56
  5118.4   637.9  5128.4  637.99  5156.5  640.17  5168.4   641.1  5186.5  642.65
  5198.4  643.67  5206.5  644.78    5216  646.08
BR D #Mann= 3
 4730.70    0.12  4991.5    0.04  5008.5    0.12
BR D Banks=4991.50,5008.50

Type RM Length L Ch R = 1 ,89650.7,544.05,544.05,544.05
XS GIS Cut Line= 3
 1964931.5173227 893422.56314008 1964666.8157421 893398.10226795
 1964447.7790315 893384.69185709
BEGIN DESCRIPTION:
Downstream Section of Bridge/Culvert/Weir
END DESCRIPTION:
#Sta/Elev= 28
  4730.7   643.6  4783.1  642.49  4840.7  640.99  4860.7  640.47  4883.1  639.89
  4933.1  636.19 4978.41  628.79  4978.5  628.77    4983  628.04  4991.5  626.65
    4994  624.55    5006  624.55  5008.5  626.65    5017  630.11 5021.39   631.9
  5021.5  631.94  5028.4  634.75  5038.4  633.55  5048.4  634.83  5058.4  635.56
  5118.4   637.9  5128.4  637.99  5156.5  640.17  5168.4   641.1  5186.5  642.65
  5198.4  643.67  5206.5  644.78    5216  646.08
#Mann= 3 , 1 , 0
 4730.70    0.12       0  4991.5    0.04       0  5008.5    0.12       0
#XS Ineff= 2 , 0
       0  4968.3   640.9  5031.6       0   641.3
Bank Sta=4991.50,5008.50
Exp/Cntr=0.5,0.3

Type RM Length L Ch R = 1 ,89106.6,606.6,606.6,606.6
XS GIS Cut Line= 3
 1965094.0459034 892897.23152182 1964795.7717349  892942.6210692
 1964585.0345507 892939.37895867
BEGIN DESCRIPTION:
South Fork Little River 178.0
END DESCRIPTION:
#Sta/Elev= 16
  4699.2  641.78  4729.2     641  4789.2   634.8  4809.2  633.53  4959.2  633.99
  4996.1  627.33  4997.6  624.33  5002.4  624.33  5003.9  627.33  5020.9  631.31
  5030.9  632.97  5040.9  634.04  5090.9  633.29  5110.9  634.58  5170.9  640.26
  5211.7  644.52
#Mann= 3 , 1 , 0
 4699.20    0.12       0  4996.1    0.04       0  5003.9    0.12       0
Bank Sta=4996.10,5003.90
Exp/Cntr=0.3,0.1

Type RM Length L Ch R = 1 ,88500.0,500,500,500
XS GIS Cut Line= 3
 1965006.5089192 892401.18861123 1964602.7109930 892441.24358113
 1964335.3920401 892498.45192703
BEGIN DESCRIPTION:
South Fork Little River 177.0
END DESCRIPTION:
#Sta/Elev= 26
  4594.2   645.7  4694.2   638.9  4804.2  631.95  4864.2  631.59  4884.2  632.88
  4894.2  632.05  4904.2  632.39  4914.2  631.62  4944.2  632.11  4974.2  631.26
  4984.2  631.77  4994.2  630.74  4996.1  626.64  4997.6  623.64  5002.4  623.64
  5003.9  626.64    5010  631.69    5020  629.54    5030  629.09    5040  631.54
    5090  631.39    5160  637.71    5180  640.07    5200  641.06    5250  642.66
  5273.4  642.84
#Mann= 3 , 1 , 0
 4594.20    0.12       0  4996.1    0.04       0  5003.9    0.12       0
Bank Sta=4996.10,5003.90
Exp/Cntr=0.3,0.1

Type RM Length L Ch R = 1 ,88000.0,500,500,500
XS GIS Cut Line= 3
 1964987.0562560  892203.4198691 1964717.7695636 892018.61435205
 1964594.7608823 891811.12449536
BEGIN DESCRIPTION:
South Fork Little River 176.0
END DESCRIPTION:
#Sta/Elev= 21
  4673.4  641.85  4803.4   633.5  4853.4  631.67  4873.4  630.23  4933.4  629.78
  4973.4  630.69  4983.4  629.57  4993.4  626.79  4996.1  625.76  4997.6  622.76
  5002.4  622.76  5003.9  625.76    5010   626.6    5030  630.01    5040  629.39
    5070   629.6    5110  632.61    5130  634.92    5170  638.16    5200  641.91
  5241.2  643.76
#Mann= 3 , 1 , 0
 4673.40    0.12       0  4996.1    0.04       0  5003.9    0.12       0
Bank Sta=4996.10,5003.90
Exp/Cntr=0.3,0.1

Type RM Length L Ch R = 1 ,87500.0,345.3,345.3,345.3
XS GIS Cut Line= 3
 1965181.5828876 891905.14570064 1964841.8217495 891741.20564028
 1964732.3175844 891692.12113352
BEGIN DESCRIPTION:
South Fork Little River 175.0
END DESCRIPTION:
#Sta/Elev= 25
  4622.8  638.42  4642.8  637.12  4712.8  635.08  4742.8  633.62  4762.8  631.96
  4772.8  631.92  4782.8   631.3  4792.8  631.55  4832.8  629.74  4892.8  629.04
  4912.8  629.68  4932.8  629.14  4962.8  630.74  4972.8  629.13  4982.8  628.36
  4996.2  625.49  4997.7  622.49  5002.4  622.49  5003.9  625.49    5010  626.77
    5020   627.9    5040  629.55    5060  633.53    5090  640.59    5120   643.6
#Mann= 3 , 1 , 0
 4622.80    0.12       0  4996.2    0.04       0  5003.9    0.12       0
Bank Sta=4996.20,5003.90
Exp/Cntr=0.3,0.1

Type RM Length L Ch R = 1 ,87154.7,601,601,601
XS GIS Cut Line= 3
 1965282.0883139 891859.75615326 1965097.2880139  891561.4819848
 1964873.5823876 891438.28178479
BEGIN DESCRIPTION:
South Fork Little River 174.0
END DESCRIPTION:
#Sta/Elev= 21
  4651.4  642.12  4821.4  637.41  4861.4  634.87  4871.4  633.51  4941.4  628.58
  4981.4  628.43  4991.4  626.84  4996.1  625.47  4997.6  622.47  5002.4  622.47
  5003.9  625.47  5032.3  626.68  5062.3  626.92  5082.3  628.94  5092.3  628.72
  5112.3  630.37  5132.3  632.77  5162.3  634.74  5172.3  636.26  5212.3  637.99
  5257.7  641.46
#Mann= 3 , 1 , 0
 4651.40    0.12       0  4996.1    0.04       0  5003.9    0.12       0
Bank Sta=4996.10,5003.90
Exp/Cntr=0.3,0.1

Type RM Length L Ch R = 1 ,86553.7,553.7,553.7,553.7
XS GIS Cut Line= 3
 1965405.2885139 891347.50269004 1965175.0986666 891195.12349528
 1964918.9719349 891068.68118474
BEGIN DESCRIPTION:
South Fork Little River 173.0
END DESCRIPTION:
#Sta/Elev= 19
  4720.7  640.97  4850.7  634.98  4930.7   631.6  4980.7  627.18  4990.7  625.32
  4996.1  622.42  4997.6  619.42  5002.4  619.42  5003.9  622.42  5006.8  622.39
  5016.8  623.42  5026.8  625.98  5036.8  626.95  5066.8  627.93  5176.8  627.33
  5196.8  629.88  5216.8  633.85  5246.8   638.4  5282.4  639.29
#Mann= 3 , 1 , 0
 4720.70    0.12       0  4996.1    0.04       0  5003.9    0.12       0
Bank Sta=4996.10,5003.90
Exp/Cntr=0.3,0.1

Type RM Length L Ch R = 1 ,86000.0,431.8,431.8,431.8
XS GIS Cut Line= 3
 1965619.2678087 891026.53374789 1965403.7268926 890761.68258501
 1965233.4566560  890530.4908373
BEGIN DESCRIPTION:
South Fork Little River 172.0
END DESCRIPTION:
#Sta/Elev= 21
  4658.5  638.05  4728.5  631.75  4818.5  627.12  4838.5  627.74  4888.5  625.08
  4908.5  625.34  4948.5  624.25  4996.1  617.65  4997.6  614.65  5002.4  614.65
  5003.9  617.65    5010  619.63    5030  623.01    5040  624.32    5050  624.92
    5060  624.59    5190  628.05    5200  628.64    5220  628.16    5270  631.79
  5287.1  633.58
#Mann= 3 , 1 , 0
 4658.50    0.12       0  4996.1    0.04       0  5003.9    0.12       0
Bank Sta=4996.10,5003.90
Exp/Cntr=0.3,0.1

Type RM Length L Ch R = 1 ,85568.2,526.8,526.8,526.8
XS GIS Cut Line= 3
 1965774.8891140 890874.15455313 1965680.8679087  890494.8276215
 1965603.0572561 890280.84832674
BEGIN DESCRIPTION:
South Fork Little River 171.0
END DESCRIPTION:
#Sta/Elev= 22
  4611.5  633.02  4661.5  630.08  4781.5  626.31  4831.5  626.88  4871.5  624.19
  4891.5  624.86  4911.5  624.17  4931.5  624.87  4971.5  622.84  4991.5  620.63
  4996.1  617.28  4997.6  614.28  5002.4  614.28  5003.9  617.28  5022.3  620.78
  5032.3  621.76  5052.3  622.81  5062.3  624.05  5132.3  628.47  5162.3  630.93
  5212.3  632.96    5230  633.23
#Mann= 3 , 1 , 0
 4611.50    0.12       0  4996.1    0.04       0  5003.9    0.12       0
Bank Sta=4996.10,5003.90
Exp/Cntr=0.3,0.1

Type RM Length L Ch R = 1 ,85041.4,489.4,489.4,489.4
XS GIS Cut Line= 3
 1966196.3634825 890258.15355305 1966005.0789614 890258.15355305
 1965606.2993666 890254.91144253
BEGIN DESCRIPTION:
South Fork Little River 170.0
END DESCRIPTION:
#Sta/Elev= 22
  4812.5  636.14  4842.5  633.43  4862.5  629.83  4892.5  626.37  4912.5  623.31
  4952.5  620.76  4992.5  621.62  4994.8   615.4  4996.3   612.4  5003.7   612.4
  5005.2   615.4  5033.8  620.07  5073.8  622.35  5093.8  626.64  5103.8  628.32
  5123.8   627.2  5213.8  629.72  5293.8  632.03  5323.8  631.27  5353.8  632.46
  5363.8  631.92  5402.6  632.95
#Mann= 3 , 1 , 0
 4812.50    0.12       0  4994.8    0.04       0  5005.2    0.12       0
Bank Sta=4994.80,5005.20
Exp/Cntr=0.3,0.1

Type RM Length L Ch R = 1 ,84552.0,447.1,447.1,447.1
XS GIS Cut Line= 3
 1966147.7318246 890063.62692145 1966112.0686088 889895.03717406
 1966084.3300262 889809.40937581
BEGIN DESCRIPTION:
South Fork Little River 169.0
END DESCRIPTION:
#Sta/Elev= 17
  4826.9  630.29  4906.9  623.39  4926.9  620.83  4946.9  619.27  4956.9  619.63
  4976.9  617.68  4986.9  617.72  4994.8  613.56  4996.3  610.56  5003.7  610.56
  5005.2  613.56  5009.2  614.61  5019.2  615.45  5029.2  618.46  5039.2  620.02
  5059.2  625.02  5089.2  631.03
#Mann= 3 , 1 , 0
 4826.90    0.12       0  4994.8    0.04       0  5005.2    0.12       0
Bank Sta=4994.80,5005.20
Exp/Cntr=0.3,0.1

Type RM Length L Ch R = 1 ,84104.9,604.9,604.9,604.9
XS GIS Cut Line= 3
 1966515.7487440 889851.53030436 1966497.8797615 889726.44742667
 1966468.7007667 889528.67868453
BEGIN DESCRIPTION:
South Fork Little River 168.0
END DESCRIPTION:
#Sta/Elev= 15
    4878  628.16    4898  626.47    4938  619.95    4958  615.65    4988  612.86
  4994.8  610.12  4996.3  607.12  5003.7  607.12  5005.2  610.12  5034.3  613.84
  5064.3  616.41  5084.3  619.63  5104.3   620.7  5184.3  626.49  5204.2  628.18
#Mann= 3 , 1 , 0
 4878.00    0.12       0  4994.8    0.04       0  5005.2    0.12       0
Bank Sta=4994.80,5005.20
Exp/Cntr=0.3,0.1

Type RM Length L Ch R = 1 ,83500.0,388,388,388
XS GIS Cut Line= 3
 1967022.9056467 889450.87597367 1966830.8466183 889287.73028571
 1966676.1771321 889160.93124719
BEGIN DESCRIPTION:
South Fork Little River 167.0
END DESCRIPTION:
#Sta/Elev= 16
    4748  624.43    4788  620.47    4828  617.25    4888  614.61    4948  609.02
    4958  608.67    4988  611.98  4994.9  606.68  4996.4  603.68  5003.7  603.68
  5005.2  606.68    5010   610.6    5020  611.32    5030  611.38    5120  617.13
    5200  624.59
#Mann= 3 , 1 , 0
 4748.00    0.12       0  4994.9    0.04       0  5005.2    0.12       0
Bank Sta=4994.90,5005.20
Exp/Cntr=0.3,0.1

Type RM Length L Ch R = 1 ,83112.0,612,612,612
XS GIS Cut Line= 3
 1967107.3965405 889279.03617398 1967013.3753352 888951.58301077
 1966778.1533784 888665.95634889
BEGIN DESCRIPTION:
South Fork Little River 166.0
END DESCRIPTION:
#Sta/Elev= 20
  4668.3  620.82  4898.3  611.14  4938.3  610.95  4978.3  608.98  4988.3  607.89
  4994.8   606.5  4996.3   603.5  5003.7   603.5  5005.2   606.5  5008.3  606.68
    5009  606.78    5019  608.12    5049   610.1    5109  610.24    5139  611.24
    5189  610.34    5279  611.71    5289  612.46    5349  620.79    5379  622.92
#Mann= 3 , 1 , 0
 4668.30    0.12       0  4994.8    0.04       0  5005.2    0.12       0
Bank Sta=4994.80,5005.20
Exp/Cntr=0.3,0.1

Type RM Length L Ch R = 1 ,82500.0,642,642,642
XS GIS Cut Line= 3
 1967528.8709090 889214.19396344 1967517.3400099 888756.03922424
 1967512.9721039 888536.08122412
BEGIN DESCRIPTION:
South Fork Little River 165.0
END DESCRIPTION:
#Sta/Elev= 19
  4541.7  618.39  4571.7  617.18  4601.7  614.07  4701.7  610.63  4711.7  610.75
  4931.7  607.67  4941.7  606.93  4951.7  607.13  4981.7  609.28  4991.7  608.26
  4994.8  606.21  4996.3  603.21  5003.7  603.21  5005.2  606.21    5010  606.82
    5030   608.4    5100  610.35    5140  615.34    5220  621.97
#Mann= 3 , 1 , 0
 4541.70    0.12       0  4994.8    0.04       0  5005.2    0.12       0
Bank Sta=4994.80,5005.20
Exp/Cntr=0.5,0.3

Type RM Length L Ch R = 1 ,81858.0,46,46,46
XS GIS Cut Line= 3
 1968037.0123726 889269.33926993 1968054.3234915 888930.53594351
 1968064.3964288 888690.80003570
BEGIN DESCRIPTION:
Upstream Section of Bridge/Culvert/Weir
END DESCRIPTION:
#Sta/Elev= 21
  4665.3  617.96  4672.2  616.26  4732.2  611.79  4772.2  609.97  4782.2  609.19
  4852.2  607.42  4942.2  607.32  4980.8   607.7    4985   602.9    5015   602.9
  5019.3   607.7    5022  607.34    5052  607.66    5062  607.33    5082  608.57
    5102  610.58    5112  612.49    5122   612.5    5162  615.42    5202  620.17
  5244.5  620.57
#Mann= 3 , 1 , 0
 4665.30    0.12       0  4980.8    0.04       0  5019.3    0.12       0
#XS Ineff= 2 , 0
       0    4964   613.7  5035.8       0   615.6
Bank Sta=4980.80,5019.30
Exp/Cntr=0.5,0.3

Type RM Length L Ch R = 3 ,81835.0,,,
BEGIN DESCRIPTION:
Wilkinson Road-TOR
Structure ID: Wilkinson Road (SFLR)-Bridge
Approximate Survey Structure
END DESCRIPTION:
Bridge Culvert--1,0,-1,-1, 0
Deck Dist Width WeirC Skew NumUp NumDn MinLoCord MaxHiCord MaxSubmerge Is_Ogee
10,26,2.6,,32,32,,,0.95,0,1,1,,
  4665.3  4672.2  4675.3  4732.2  4765.3  4772.2  4782.2  4785.3  4805.3  4852.2
  4942.2 4974.11  4974.2    4980  4980.8    4985    5015  5019.3    5020    5022
 5025.59  5025.7    5052    5062    5082    5102    5112    5122    5162  5184.5
    5202  5244.5
  617.96  617.45  617.22  615.76  614.91  614.64  614.25  614.13  613.72   614.1
  614.84   615.1   615.1  615.15  615.15  615.19  615.43  615.47  615.48  615.49
  615.52  615.52  615.74  615.82  615.98  616.15  616.23  616.31  616.64   618.1
  620.18  620.57
  617.96  616.26  616.03  611.79  610.28  609.97  609.19  609.11  608.61  607.42
  607.32  607.63   612.7  612.75  612.75  612.79  613.03  613.07  613.08  613.09
  613.12  607.38  607.66  607.33  608.57  610.58  612.49   612.5  615.42  618.09
  620.17  620.57
  4665.3  4672.2  4675.3  4732.2  4765.3  4772.2  4782.2  4785.3  4805.3  4852.2
  4942.2 4974.11  4974.2    4980  4980.8    4985    5015  5019.3    5020    5022
 5025.59  5025.7    5052    5062    5082    5102    5112    5122    5162  5184.5
    5202  5244.5
  617.96  617.45  617.22  615.76  614.91  614.64  614.25  614.13  613.72   614.1
  614.84   615.1   615.1  615.15  615.15  615.19  615.43  615.47  615.48  615.49
  615.52  615.52  615.74  615.82  615.98  616.15  616.23  616.31  616.64   618.1
  620.18  620.57
  617.71  616.01  615.78  611.54  610.03  609.72  608.94  608.86  608.36  607.17
  607.07  607.38  612.45   612.5   612.5  612.54  612.78  612.82  612.83  612.84
  612.87  607.13  607.41  607.08  608.32  610.33  612.24  612.25  615.17  617.84
  619.92  620.32
Pier Skew, UpSta & Num, DnSta & Num=,4984.0, 2 ,4984.0, 2 , 0 , 0 , 0 ,,
       1       1
  602.47  613.79
       1       1
  602.22  613.54
Pier Skew, UpSta & Num, DnSta & Num=,4992.0, 2 ,4992.0, 2 , 0 , 0 , 0 ,,
       1       1
   601.9  613.85
       1       1
  601.65   613.6
Pier Skew, UpSta & Num, DnSta & Num=,5000.0, 2 ,5000.0, 2 , 0 , 0 , 0 ,,
       1       1
   601.9  613.91
       1       1
  601.65  613.66
Pier Skew, UpSta & Num, DnSta & Num=,5008.0, 2 ,5008.0, 2 , 0 , 0 , 0 ,,
       1       1
   601.9  613.98
       1       1
  601.65  613.73
Pier Skew, UpSta & Num, DnSta & Num=,5016.0, 2 ,5016.0, 2 , 0 , 0 , 0 ,,
       1       1
  602.46  614.04
       1       1
  602.21  613.79
Abutment Skew #Up #Dn=, 2 , 2
 4974.00 4980.00
  612.70  607.69
 4974.00 4980.00
  612.45  607.44
Abutment Skew #Up #Dn=, 2 , 2
 5020.00 5025.79
  607.61  613.12
 5020.00 5025.79
  607.36  612.87
BR Coef= 1 , 1 , 0 ,1.25, 0 ,,,0.8,0,2,0,
Wspro=,,,, 1 ,,,, 0 ,,,, 0 ,,,,-1 ,-1 ,-1 , 0 , 0 , 0 , 0 , 0
BC Design=,, 0 ,, 0 ,,,,,,
BR U #Sta/Elev= 32
  4665.3  617.96  4672.2  616.26  4675.3  616.03  4732.2  611.79  4765.3  610.28
  4772.2  609.97  4782.2  609.19  4785.3  609.11  4805.3  608.61  4852.2  607.42
  4942.2  607.32 4974.11  607.63  4974.2  607.64    4980  607.69  4980.8   607.7
    4985   602.9    5015   602.9  5019.3   607.7    5020  607.61    5022  607.34
 5025.59  607.38  5025.7  607.38    5052  607.66    5062  607.33    5082  608.57
    5102  610.58    5112  612.49    5122   612.5    5162  615.42  5184.5  618.09
    5202  620.17  5244.5  620.57
BR U #Mann= 3
 4665.30    0.12  4980.8    0.04  5019.3    0.12
BR U Banks=4980.80,5019.30
BR D #Sta/Elev= 32
  4665.3  617.71  4672.2  616.01  4675.3  615.78  4732.2  611.54  4765.3  610.03
  4772.2  609.72  4782.2  608.94  4785.3  608.86  4805.3  608.36  4852.2  607.17
  4942.2  607.07 4974.11  607.38  4974.2  607.39    4980  607.44  4980.8  607.45
    4985  602.65    5015  602.65  5019.3  607.45    5020  607.36    5022  607.09
 5025.59  607.13  5025.7  607.13    5052  607.41    5062  607.08    5082  608.32
    5102  610.33    5112  612.24    5122  612.25    5162  615.17  5184.5  617.84
    5202  619.92  5244.5  620.32
BR D #Mann= 3
 4665.30    0.12  4980.8    0.04  5019.3    0.12
BR D Banks=4980.80,5019.30

Type RM Length L Ch R = 1 ,81812.0,312,312,312
XS GIS Cut Line= 3
 1968082.9910707 889270.73902734 1968100.3021896 888931.93570092
 1968110.3751269 888692.19979311
BEGIN DESCRIPTION:
Downstream Section of Bridge/Culvert/Weir
END DESCRIPTION:
#Sta/Elev= 21
  4665.3  617.68  4672.2  615.98  4732.2  611.51  4772.2  609.69  4782.2  608.91
  4852.2  607.14  4942.2  607.04  4980.8  607.42    4985  602.62    5015  602.62
  5019.3  607.42    5022  607.06    5052  607.38    5062  607.05    5082  608.29
    5102   610.3    5112  612.21    5122  612.22    5162  615.14    5202  619.89
  5244.5  620.29
#Mann= 3 , 1 , 0
 4665.30    0.12       0  4980.8    0.04       0  5019.3    0.12       0
#XS Ineff= 2 , 0
       0    4964   613.7  5035.8       0   615.6
Bank Sta=4980.80,5019.30
Exp/Cntr=0.5,0.3

Type RM Length L Ch R = 1 ,81500.0,500,500,500
XS GIS Cut Line= 3
 1968514.4725091 889149.35175291 1968369.9296361 888809.86639011
 1968330.1334716 888718.12402223
BEGIN DESCRIPTION:
South Fork Little River 163.0
END DESCRIPTION:
#Sta/Elev= 18
    4631  617.12    4671   613.1    4681  611.61    4811  605.01    4881  606.12
    4921  605.24    4941  606.44    4981  606.92    4991  606.54  4994.8  604.82
  4996.3  601.82  5003.7  601.82  5005.2  604.82    5010  605.55    5040  609.63
    5050  610.49    5080  615.45    5100  620.38
#Mann= 3 , 1 , 0
 4631.00    0.12       0  4994.8    0.04       0  5005.2    0.12       0
Bank Sta=4994.80,5005.20
Exp/Cntr=0.3,0.1

Type RM Length L Ch R = 1 ,81000.0,697.4,697.4,697.4
XS GIS Cut Line= 3
 1968913.2521039 888799.20381602 1968781.9650777  888549.9559714
 1968670.0938144 888342.06623175
BEGIN DESCRIPTION:
South Fork Little River 162.0
END DESCRIPTION:
#Sta/Elev= 22
  4718.3  617.28  4738.3  616.03  4758.3  615.48  4788.3  613.31  4808.3  613.19
  4868.3  606.82  4878.3  606.06  4888.3  605.82  4908.3  605.92  4988.3  604.31
  4994.8  603.53  4996.3  600.53  5003.7  600.53  5005.2  603.53    5010  604.26
    5050  605.41    5110     605    5150   610.9    5160  611.92    5180  615.15
    5200  616.46  5236.1   621.5
#Mann= 3 , 1 , 0
 4718.30    0.12       0  4994.8    0.04       0  5005.2    0.12       0
Bank Sta=4994.80,5005.20
Exp/Cntr=0.3,0.1

Type RM Length L Ch R = 1 ,80302.6,853.3,853.3,853.3
XS GIS Cut Line= 3
 1969123.9892881 888841.35125287 1969240.7052671 888474.99276334
 1969389.8423513 887940.04452643
BEGIN DESCRIPTION:
South Fork Little River 161.0
END DESCRIPTION:
#Sta/Elev= 21
  4617.8   617.2  4647.8  616.99  4727.8  612.17  4777.8  606.99  4807.8  605.01
  4837.8     604  4877.8  604.32  4897.8  603.52  4927.8  603.63  4992.4  601.76
  4993.9  598.76  5006.2  598.76  5007.7  601.76  5012.3     603  5072.3  603.61
  5112.3  605.59  5142.3  605.53  5162.3  606.37  5272.3  606.12  5392.3  609.48
  5557.6  617.17
#Mann= 3 , 1 , 0
 4617.80    0.12       0  4992.4    0.04       0  5007.7    0.12       0
Bank Sta=4992.40,5007.70
Exp/Cntr=0.3,0.1

Type RM Length L Ch R = 1 ,79449.3,370.3,370.3,370.3
XS GIS Cut Line= 3
 1970010.7065172 888625.10248073  1969830.769383 888160.50804225
 1969645.8478064 887887.15974320
BEGIN DESCRIPTION:
South Fork Little River 159.0
END DESCRIPTION:
#Sta/Elev= 21
  4508.3   612.6  4538.3  609.33  4608.3  605.33  4638.3  604.12  4808.3  602.34
  4818.3  602.83  4898.3  601.77  4958.3  600.11  4988.3  599.97  4992.4  597.62
  4993.9  594.62  5006.2  594.62  5007.7  597.62  5016.5  598.62  5066.5  600.53
  5146.5  601.01  5166.5  600.08  5226.5  601.33  5266.5  606.48  5296.5  611.36
  5336.5  616.23
#Mann= 3 , 1 , 0
 4508.30    0.14       0  4992.4   0.045       0  5007.7    0.15       0
Bank Sta=4992.40,5007.70
Exp/Cntr=0.3,0.1

Type RM Length L Ch R = 1 ,79079.0,579,579,579
XS GIS Cut Line= 3
 1970264.8879825  888596.5719081 1970168.9215109 888090.80266592
 1969969.2075024 887515.00383637
BEGIN DESCRIPTION:
South Fork Little River 158.0
END DESCRIPTION:
#Sta/Elev= 23
    4488  615.46    4548   611.9    4578  608.88    4678  604.34    4698  603.35
    4788  601.92    4808  601.62    4838  601.82    4948  600.27    4968  600.57
    4988  598.73  4992.3  596.74  4993.8  593.74  5006.1  593.74  5007.6  596.74
  5012.8  599.06  5142.8  601.29  5252.8  601.73  5322.8  604.13  5422.8  605.72
  5502.8  607.01  5562.8  608.06  5612.2  608.55
#Mann= 3 , 1 , 0
 4488.00    0.14       0  4992.3   0.045       0  5007.6    0.15       0
Bank Sta=4992.30,5007.60
Exp/Cntr=0.3,0.1

Type RM Length L Ch R = 1 ,78500.0,500,500,500
XS GIS Cut Line= 3
 1970630.5980499 887958.52455643 1970497.4294963 887864.26603231
 1969979.5822561 887429.41211847
BEGIN DESCRIPTION:
South Fork Little River 157.0
END DESCRIPTION:
#Sta/Elev= 27
  4836.8  614.07  4886.8  610.83  4896.8  609.64  4936.8  602.87  4956.8  598.96
  4966.8  598.16  4976.8  598.72  4986.8  598.39  4992.3  596.03  4993.8  593.03
  5006.1  593.03  5007.6  596.03    5010  596.06    5020  596.96    5030  599.19
    5040  599.46    5050  598.46    5060  598.58    5070  599.85    5080  600.27
    5180  600.04    5290  600.95    5300  600.58    5370  602.52    5440  605.65
    5640  608.02  5676.2  608.81
#Mann= 3 , 1 , 0
 4836.80    0.14       0  4992.3   0.045       0  5007.6    0.15       0
Bank Sta=4992.30,5007.60
Exp/Cntr=0.3,0.1

Type RM Length L Ch R = 1 ,78000.0,500,500,500
XS GIS Cut Line= 3
 1970788.5028501 887502.56447884 1970591.5583274 887451.32183653
 1969904.3652919  887227.1044216
BEGIN DESCRIPTION:
South Fork Little River 156.0
END DESCRIPTION:
#Sta/Elev= 26
  4796.5  617.93  4856.5  612.68  4886.5  608.56  4926.5  600.57  4946.5  598.48
  4956.5  598.29  4992.4  596.01  4993.9  593.01  5006.2  593.01  5007.7  596.01
    5010  596.31    5030  598.61    5050  598.74    5090  596.84    5110  597.69
    5120     597    5190  600.78    5330  603.64    5360  603.79    5410  605.09
    5440  604.87    5530  606.66    5600     609    5650  610.01    5670  611.35
  5722.9  613.51
#Mann= 3 , 1 , 0
 4796.50    0.14       0  4992.4   0.045       0  5007.7    0.15       0
Bank Sta=4992.40,5007.70
Exp/Cntr=0.3,0.1

Type RM Length L Ch R = 1 ,77500.0,500,500,500
XS GIS Cut Line= 3
 1970842.4748164 887154.40646446 1970624.8639840 887082.75788726
 1970028.8623361 886889.92492682
BEGIN DESCRIPTION:
South Fork Little River 155.0
END DESCRIPTION:
#Sta/Elev= 23
  4770.9  612.07  4780.9   610.6  4810.9  607.89  4830.9  605.13  4840.9  603.33
  4880.9  599.44  4990.9  596.67  4992.4  595.98  4993.9  592.98  5006.2  592.98
  5007.7  595.98    5010   596.5    5030  597.39    5140  599.58    5160  600.78
    5220   601.7    5250   602.6    5340  604.04    5460  605.11    5530  606.96
    5560  608.46    5580  610.47  5626.4  613.25
#Mann= 3 , 1 , 0
 4770.90    0.14       0  4992.4   0.045       0  5007.7    0.15       0
Bank Sta=4992.40,5007.70
Exp/Cntr=0.3,0.1

Type RM Length L Ch R = 1 ,77000.0,526.45,526.45,526.45
XS GIS Cut Line= 3
 1970958.2699023 886747.64125846 1970780.7151224  886629.9731112
 1970353.0733888 886332.28191622
BEGIN DESCRIPTION:
South Fork Little River 154.0
END DESCRIPTION:
#Sta/Elev= 22
    4787  615.55    4827  609.56    4847  607.72    4867  606.89    4927  600.27
    4987  595.79  4992.4  594.74  4993.9  591.74  5006.2  591.74  5007.7  594.74
    5010  594.74    5060   597.1    5080  596.52    5140   596.6    5160   595.8
    5200  595.74    5280  597.34    5290  596.93    5360  597.65    5440  601.95
    5450   603.4  5521.1  607.11
#Mann= 3 , 1 , 0
 4787.00    0.14       0  4992.4   0.045       0  5007.7    0.15       0
Bank Sta=4992.40,5007.70
Exp/Cntr=0.5,0.3

Type RM Length L Ch R = 1 ,76473.6,63.5,63.5,63.5
XS GIS Cut Line= 3
 1971136.1832219 886508.68109082 1970918.6118617 886200.45499717
 1970538.9825896 885784.67055630
BEGIN DESCRIPTION:
Upstream Section of Bridge/Culvert/Weir
END DESCRIPTION:
#Sta/Elev= 26
  4627.7  605.49  4684.4  602.73  4694.4  603.02  4814.4  599.73  4834.4  599.78
  4874.4   598.7  4904.4  597.46  4954.4  598.53    4977  593.14  4978.5  590.14
  5021.5  590.14    5023  593.14  5050.3  596.25  5060.3  596.88  5100.3  595.62
  5160.3  596.95  5180.3  596.05  5210.3  596.08  5220.3  596.59  5430.3   597.3
  5470.3  598.83  5500.3   598.1  5510.3  598.35  5520.3  599.52  5550.3  604.42
    5568  606.08
#Mann= 3 , 1 , 0
 4627.70    0.14       0    4977   0.045       0    5023    0.15       0
#XS Ineff= 2 , 0
       0  4968.5   601.3  5031.5       0   601.2
Bank Sta=4977.00,5023.00
Exp/Cntr=0.5,0.3

Type RM Length L Ch R = 2 ,76441.8,,,
BEGIN DESCRIPTION:
Walnut Grove Ch Road (SFLR)-TOR
Structure ID: Walnut Grove Ch Road (SFLR)-Culvert
Approximate Survey Structure
END DESCRIPTION:
Bridge Culvert--1,0,-1,-1, 0
Deck Dist Width WeirC Skew NumUp NumDn MinLoCord MaxHiCord MaxSubmerge Is_Ogee
10,43.5,3,,35,35,,,0.95,0,1,1,,
  4627.7  4634.4  4667.7  4684.4  4694.4  4737.7  4787.7  4814.4  4834.4  4857.7
  4874.4  4904.4  4954.4    4977  4978.5  5021.5    5023  5050.3  5060.3  5100.3
  5160.3  5180.3  5210.3  5220.3    5305  5430.3    5435  5470.3    5495  5500.3
  5510.3  5520.3  5522.6  5550.3    5568
  605.45   605.1  603.92  603.51  603.27  602.22  601.83  601.63  601.48  601.31
  601.31   601.3  601.29  601.28  601.28  601.27  601.27  601.27  601.26  601.26
  601.24  601.24  601.23  601.23  601.21  601.68   601.7  602.37  602.84  602.89
  602.99  603.09  603.11  604.38  606.04
  605.45  605.08  603.49  602.69  602.98  601.79  600.42  599.69  599.74  599.11
  598.66  597.42  598.49   593.1   590.1   590.1   593.1  596.21  596.84  595.58
  596.91  596.01  596.04  596.55  596.84  597.26  597.44  598.79  598.19  598.06
  598.31  599.48  599.86  604.38  606.04
  4627.7  4634.4  4667.7  4684.4  4694.4  4737.7  4787.7  4814.4  4834.4  4857.7
  4874.4  4904.4  4954.4    4977  4978.5  5021.5    5023  5050.3  5060.3  5100.3
  5160.3  5180.3  5210.3  5220.3    5305  5430.3    5435  5470.3    5495  5500.3
  5510.3  5520.3  5522.6  5550.3    5568
  605.34   605.1  603.92  603.51  603.27  602.22  601.83  601.63  601.48  601.31
  601.31   601.3  601.29  601.28  601.28  601.27  601.27  601.27  601.26  601.26
  601.24  601.24  601.23  601.23  601.21  601.68   601.7  602.37  602.84  602.89
  602.99  603.09  603.11  604.27  605.93
  605.23  604.86  603.27  602.47  602.76  601.57   600.2  599.47  599.52  598.89
  598.44   597.2  598.27  592.88  589.88  589.88  592.88  595.99  596.62  595.36
  596.69  595.79  595.82  596.33  596.62  597.04  597.22  598.57  597.97  597.84
  598.09  599.26  599.64  604.16  605.82
BR Coef= 1 , 0 , 0 ,1.25, 0 ,,,0.8,-1,2,0,
Wspro=,,,, 1 ,,,, 0 ,,,, 0 ,,,,-1 ,-1 ,-1 , 0 , 0 , 0 , 0 , 0
Culvert=2,8.0,10.0,43.5,0.015,0.4,1.0,8,1,590.10,4983.50,589.88,4983.50,Culvert #1  ,0,10
Culvert=2,8.0,10.0,43.5,0.015,0.4,1.0,8,1,590.10,4994.50,589.88,4994.50,Culvert #2  ,0,10
Culvert=2,8.0,10.0,43.5,0.015,0.4,1.0,8,1,590.10,5005.50,589.88,5005.50,Culvert #3  ,0,10
Culvert=2,8.0,10.0,43.5,0.015,0.4,1.0,8,1,590.10,5016.50,589.88,5016.50,Culvert #4  ,0,10
BC Design=,, 0 ,, 0 ,,,,,,
BR U #Sta/Elev= 35
  4627.7  605.45  4634.4  605.08  4667.7  603.49  4684.4  602.69  4694.4  602.98
  4737.7  601.79  4787.7  600.42  4814.4  599.69  4834.4  599.74  4857.7  599.11
  4874.4  598.66  4904.4  597.42  4954.4  598.49    4977   593.1  4978.5   590.1
  5021.5   590.1    5023   593.1  5050.3  596.21  5060.3  596.84  5100.3  595.58
  5160.3  596.91  5180.3  596.01  5210.3  596.04  5220.3  596.55    5305  596.84
  5430.3  597.26    5435  597.44  5470.3  598.79    5495  598.19  5500.3  598.06
  5510.3  598.31  5520.3  599.48  5522.6  599.86  5550.3  604.38    5568  606.04
BR U #Mann= 3
 4627.70    0.14    4977   0.045    5023    0.15
BR U Banks=4977.00,5023.00
BR D #Sta/Elev= 35
  4627.7  605.23  4634.4  604.86  4667.7  603.27  4684.4  602.47  4694.4  602.76
  4737.7  601.57  4787.7   600.2  4814.4  599.47  4834.4  599.52  4857.7  598.89
  4874.4  598.44  4904.4   597.2  4954.4  598.27    4977  592.88  4978.5  589.88
  5021.5  589.88    5023  592.88  5050.3  595.99  5060.3  596.62  5100.3  595.36
  5160.3  596.69  5180.3  595.79  5210.3  595.82  5220.3  596.33    5305  596.62
  5430.3  597.04    5435  597.22  5470.3  598.57    5495  597.97  5500.3  597.84
  5510.3  598.09  5520.3  599.26  5522.6  599.64  5550.3  604.16    5568  605.82
BR D #Mann= 3
 4627.70    0.14    4977   0.045    5023    0.15
BR D Banks=4977.00,5023.00

Type RM Length L Ch R = 1 ,76410.1,292.65,292.65,292.65
XS GIS Cut Line= 3
 1971179.5030453 886462.25218923 1970961.9316850 886154.02609558
  1970582.302413 885738.24165471
BEGIN DESCRIPTION:
Downstream Section of Bridge/Culvert/Weir
END DESCRIPTION:
#Sta/Elev= 26
  4627.7  605.22  4684.4  602.46  4694.4  602.75  4814.4  599.46  4834.4  599.51
  4874.4  598.43  4904.4  597.19  4954.4  598.26    4977  592.87  4978.5  589.87
  5021.5  589.87    5023  592.87  5050.3  595.98  5060.3  596.61  5100.3  595.35
  5160.3  596.68  5180.3  595.78  5210.3  595.81  5220.3  596.32  5430.3  597.03
  5470.3  598.56  5500.3  597.83  5510.3  598.08  5520.3  599.25  5550.3  604.15
    5568  605.81
#Mann= 3 , 1 , 0
 4627.70    0.14       0    4977   0.045       0    5023    0.15       0
#XS Ineff= 2 , 0
       0  4968.5   601.3  5031.5       0   601.2
Bank Sta=4977.00,5023.00
Exp/Cntr=0.5,0.3

Type RM Length L Ch R = 1 ,76117.4,617.4,617.4,617.4
XS GIS Cut Line= 3
 1971481.3278521 886225.94069094 1971048.1818857 885896.54226142
 1970679.8859453 885474.58730984
BEGIN DESCRIPTION:
South Fork Little River 152.0
END DESCRIPTION:
#Sta/Elev= 29
  4451.1  607.27  4481.1  605.24  4641.1  602.65  4661.1  601.12  4681.1  600.45
  4711.1  598.85  4731.1   598.8  4761.1  597.39  4771.1  597.75  4801.1  596.71
  4891.1  595.84  4971.1  596.94  4981.1  596.57  4992.4  592.62  4993.9  589.62
  5006.2  589.62  5007.7  592.62  5025.3  596.14  5195.3  594.27  5215.3  595.19
  5245.3  594.65  5255.3  595.08  5405.3  595.63  5445.3  594.26  5485.3  595.14
  5505.3  597.35  5525.3  605.35  5535.3  608.14  5555.3  612.16
#Mann= 3 , 1 , 0
 4451.10    0.12       0  4992.4   0.045       0  5007.7    0.14       0
Bank Sta=4992.40,5007.70
Exp/Cntr=0.3,0.1

Type RM Length L Ch R = 1 ,75500.0,402.6,402.6,402.6
XS GIS Cut Line= 3
 1971636.9491574 886028.82037092 1971108.4100420 885449.08167737
 1970861.4363194 885222.18327186
BEGIN DESCRIPTION:
South Fork Little River 151.0
END DESCRIPTION:
#Sta/Elev= 30
  4215.5  606.36  4285.5  601.15  4395.5  597.96  4475.5  597.65  4525.5  595.78
  4565.5  595.34  4625.5  595.31  4645.5  594.32  4675.5  595.15  4695.5  594.07
  4835.5  594.21  4845.5  595.15  4885.5  594.25  4905.5  595.38  4965.5  594.46
  4985.5  592.23  4992.4  590.16  4993.9  587.16  5006.2  587.16  5007.7  590.16
    5010  591.96    5020  593.77    5050  594.11    5060  593.31    5070  593.05
    5100  592.97    5130     594    5250  595.02    5310  598.84  5335.4   603.3
#Mann= 3 , 1 , 0
 4215.50    0.12       0  4992.4   0.045       0  5007.7    0.14       0
Bank Sta=4992.40,5007.70
Exp/Cntr=0.3,0.1

Type RM Length L Ch R = 1 ,75097.4,698.6,698.6,698.6
XS GIS Cut Line= 3
 1971966.3475869 885696.82825298 1971411.2982647 885196.24638765
 1971197.0258993 884972.23436922
BEGIN DESCRIPTION:
South Fork Little River 150.0
END DESCRIPTION:
#Sta/Elev= 30
  4251.6  602.53  4291.6  599.19  4351.6  596.39  4481.6  595.09  4491.6  594.18
  4541.6  592.77  4651.6  592.84  4701.6  591.79  4721.6  592.54  4741.6  591.74
  4781.6  592.95  4811.6  592.46  4951.6  592.75  4971.6  593.71  4981.6  593.22
  4991.6  589.72  4992.4  588.33  4993.9  585.33  5006.2  585.33  5007.7  588.33
    5009  590.97    5019  593.33    5049  593.11    5069  592.15    5109  593.01
    5179  592.07    5199  592.55    5259  599.14    5279  603.36    5309  607.69
#Mann= 3 , 1 , 0
 4251.60    0.12       0  4992.4   0.045       0  5007.7    0.14       0
Bank Sta=4992.40,5007.70
Exp/Cntr=0.3,0.1

Type RM Length L Ch R = 1 ,74398.8,398.8,398.8,398.8
XS GIS Cut Line= 3
 1972090.8446311 885538.61325927 1971927.4422606 884812.38050128
 1971904.3329009 884633.80817650
BEGIN DESCRIPTION:
South Fork Little River 149.0
END DESCRIPTION:
#Sta/Elev= 30
  4255.3  600.41  4285.3  599.74  4345.3  596.11  4355.3  594.96  4395.3  593.31
  4445.3  591.74  4475.3  591.75  4505.3  590.47  4545.3  590.99  4555.3  590.67
  4605.3  591.75  4735.3  591.27  4755.3  590.49  4825.3  591.02  4835.3  590.43
  4845.3  590.94  4855.3   590.5  4915.3  591.73  4935.3  591.34  4955.3  591.97
  4965.3  592.71  4992.4  586.96  4993.9  583.96  5006.2  583.96  5007.7  586.96
  5009.7  592.61  5019.7  594.63  5069.7  597.57  5119.7  603.85  5179.7   613.8
#Mann= 3 , 1 , 0
 4255.30    0.12       0  4992.4   0.045       0  5007.7    0.14       0
Bank Sta=4992.40,5007.70
Exp/Cntr=0.3,0.1

Type RM Length L Ch R = 1 ,74000.0,566.6,566.6,566.6
XS GIS Cut Line= 3
 1972448.7736333 885030.25032868 1972253.6581634 884647.02899666
 1972174.0014179 884519.92877979
BEGIN DESCRIPTION:
South Fork Little River 148.0
END DESCRIPTION:
#Sta/Elev= 28
    4570   602.7    4610  599.37    4620  598.06    4640  592.55    4650  591.31
    4680  589.46    4810  589.79    4820  588.96    4830  589.67    4840  589.87
    4850  589.51    4880  590.61    4910  588.47    4930  588.95    4960  590.03
    4970  591.05    4980   591.2    4990  590.48  4992.4  586.28  4993.9  583.28
  5006.2  583.28  5007.7  586.28    5010  587.93    5030  590.56    5080  592.57
    5110  595.34    5120  596.99    5150  605.91
#Mann= 3 , 1 , 0
 4570.00    0.12       0  4992.4   0.045       0  5007.7    0.14       0
Bank Sta=4992.40,5007.70
Exp/Cntr=0.3,0.1

Type RM Length L Ch R = 1 ,73433.4,508.5,508.5,508.5
XS GIS Cut Line= 3
 1972793.7341933  884887.5974655 1972705.5487870 884480.38838334
 1972711.6171937 884400.71208831
BEGIN DESCRIPTION:
South Fork Little River 147.0
END DESCRIPTION:
#Sta/Elev= 20
  4580.8  598.89  4650.8  592.81  4690.8  591.16  4710.8  589.67  4730.8  588.99
  4790.8   589.7  4810.8  588.87  4830.8  589.17  4850.8  588.32  4930.8  589.05
  4970.8  587.47  4990.8  586.05  4992.3     584  4993.8     581  5006.1     581
  5007.6     584  5017.4   589.1  5027.4  592.07  5047.4   599.4  5077.4  604.22
#Mann= 3 , 1 , 0
 4580.80    0.12       0  4992.3   0.045       0  5007.6    0.14       0
Bank Sta=4992.30,5007.60
Exp/Cntr=0.3,0.1

Type RM Length L Ch R = 1 ,72924.9,516.9,516.9,516.9
XS GIS Cut Line= 3
 1973250.2233555 884783.84992865 1973146.4758187 884433.70199176
 1973066.0714776 884093.92880855
BEGIN DESCRIPTION:
South Fork Little River 146.0
END DESCRIPTION:
#Sta/Elev= 24
  4639.6  602.17  4679.6  596.45  4689.6  594.27  4699.6  592.65  4779.6   588.4
  4919.6  588.15  4929.6  587.66  4959.6  588.46  4969.6   588.3  4979.6  587.48
  4991.9  583.44  4993.4  580.44  5006.7  580.44  5008.2  583.44  5024.8  586.67
  5044.8  587.15  5084.8  588.47  5144.8  587.44  5194.8  587.85  5244.8  590.68
  5274.8  593.71  5304.8  597.63  5314.8  599.56    5354   602.4
#Mann= 3 , 1 , 0
 4639.60    0.12       0  4991.9   0.045       0  5008.2    0.14       0
Bank Sta=4991.90,5008.20
Exp/Cntr=0.3,0.1

Type RM Length L Ch R = 1 ,72408.0,655.85,655.85,655.85
XS GIS Cut Line= 3
 1973870.1148882 884316.98601279 1973556.2785892 884169.14577278
 1973439.3834219 884045.74714317
BEGIN DESCRIPTION:
South Fork Little River 145.0
END DESCRIPTION:
#Sta/Elev= 23
  4656.9  607.33  4726.9  601.75  4746.9  600.16  4776.9  597.53  4806.9  592.93
  4826.9  588.59  4836.9  587.18  4876.9  586.34  4886.9  587.03  4916.9  587.07
  4976.9  585.44  4991.8   583.2  4993.3   580.2  5006.6   580.2  5008.1   583.2
  5013.8  585.57  5023.8  587.02  5033.8  587.09  5043.8  589.37  5113.8  600.15
  5123.8  601.26  5163.8  602.99  5173.8  604.25
#Mann= 3 , 1 , 0
 4656.90    0.12       0  4991.8   0.045       0  5008.1    0.14       0
Bank Sta=4991.80,5008.10
Exp/Cntr=0.5,0.3

Type RM Length L Ch R = 1 ,71752.2,40.5,40.5,40.5
XS GIS Cut Line= 3
 1974201.1082624 883880.34643121 1973912.8082914 883691.97706871
 1973617.7765115 883576.13636983
BEGIN DESCRIPTION:
Upstream Section of Bridge/Culvert/Weir
END DESCRIPTION:
#Sta/Elev= 24
  4656.8  596.33  4777.5  590.04  4817.5  587.15  4837.5  587.68  4867.5  586.03
  4877.5  586.23  4887.5   585.9  4897.5   586.6  4917.5  588.84  4927.5  588.82
  4977.3  584.94  4987.5  584.82    4990   583.4    4992   579.9    5008   579.9
    5010   583.4  5011.7  582.83  5021.7  586.46  5031.7  587.86  5061.7  588.43
  5071.7  589.28  5081.7  590.77  5131.7   594.6  5318.1  600.64
#Mann= 3 , 1 , 0
 4656.80    0.12       0    4990   0.045       0    5010    0.14       0
#XS Ineff= 2 , 0
       0  4967.3     588  5032.6       0   590.8
Bank Sta=4990.00,5010.00
Exp/Cntr=0.5,0.3
