HEC-RAS study SOUTH FORK.PRJ: South Fork

--- SOUTH FORK.g01 (geometry) --- (continued)

Type RM Length L Ch R = 1 ,26906.6,654.9,654.9,654.9
XS GIS Cut Line= 3
      1892573.96       764063.14      1892792.67       764004.93
      1892887.58       763978.68
BEGIN DESCRIPTION:
South Fork 44.0
END DESCRIPTION:
#Sta/Elev= 24
  4771.9  523.41  4832.1     521  4846.1  519.72  4851.4  519.78    4862  519.73
  4874.8  517.81  4907.4  519.04  4908.7  518.73  4930.1  511.14  4952.3  509.93
  4986.2  504.14  4989.2  500.14 5010.65  500.14 5013.65  504.14  5018.9  504.66
  5021.5  505.31    5037  513.27  5042.6  513.94    5051  517.02  5058.7  518.52
  5067.5  519.64  5069.3  520.32  5086.1  522.12  5096.7  523.96
#Mann= 3 , 1 , 0
 4771.90    0.13       0  4986.2    0.05       0 5013.65    0.12       0
Bank Sta=4986.20,5013.65
Exp/Cntr=0.3,0.1

Type RM Length L Ch R = 1 ,26251.7,549.6,549.6,549.6
XS GIS Cut Line= 3
      1892740.14       764589.50      1892785.25       764504.18
      1892949.54       764173.78
BEGIN DESCRIPTION:
South Fork 43.0
END DESCRIPTION:
#Sta/Elev= 30
  4903.5  522.95  4905.7  521.96  4916.2  519.29  4931.5  515.64  4939.7  514.11
  4954.6  512.12  4973.3  510.72  4973.8  510.59  4986.2  503.92 4986.35  503.64
 4989.35  499.64  5010.8  499.64  5013.8  503.64  5020.6  504.94  5022.8  508.21
  5045.3  507.38  5063.8     507  5069.4  507.07    5083  508.15  5110.5  509.43
  5120.5  509.66  5130.9  509.12  5144.3  508.75  5159.6  508.59  5178.7  508.66
  5223.6  509.23  5264.1  511.04  5281.5  512.61  5300.5  514.74    5369  523.39
#Mann= 3 , 1 , 0
 4903.50    0.13       0 4986.35    0.05       0  5013.8    0.12       0
Bank Sta=4986.35,5013.80
Exp/Cntr=0.3,0.1

Type RM Length L Ch R = 1 ,25702.1,784.2,784.2,784.2
XS GIS Cut Line= 3
      1892911.71       764728.22      1893210.38       764694.19
      1893333.64       764683.76
BEGIN DESCRIPTION:
South Fork 42.0
END DESCRIPTION:
#Sta/Elev= 30
  4699.4  522.56  4713.5  519.35  4729.4  517.01  4734.7  515.99  4745.1  513.15
  4752.8  511.85  4776.1   509.4  4784.5  509.15  4797.2  507.97  4818.9  507.45
  4834.1  507.28  4839.3  507.79    4890   507.2  4929.5  507.37  4947.2  506.57
  4967.8  504.55  4975.5  503.15 4986.35  502.29 4989.35  498.29  5010.8  498.29
  5013.8  502.29  5015.7  503.71  5020.9  504.54  5030.5  508.94  5051.5  513.32
  5072.5  516.76  5091.8  518.08  5107.5  519.56  5121.1  521.79  5123.7  522.47
#Mann= 3 , 1 , 0
 4699.40    0.14       0 4986.35    0.05       0  5013.8    0.13       0
Bank Sta=4986.35,5013.80
Exp/Cntr=0.3,0.1

Type RM Length L Ch R = 1 ,24917.9,428.1,428.1,428.1
XS GIS Cut Line= 3
      1893272.45       765436.89      1893374.75       765349.88
      1893516.71       765213.44
BEGIN DESCRIPTION:
South Fork 41.0
END DESCRIPTION:
#Sta/Elev= 21
  4865.7  520.45  4926.6  512.58    4928  512.21    4938  510.03  4950.7  508.17
    4971  505.94  4972.8  505.85  4973.8  505.51 4986.35  502.22 4989.35  498.22
  5010.8  498.22  5013.8  502.22  5043.5  503.74  5055.6   505.5  5079.5  506.99
  5099.6  509.33  5108.7  510.82  5113.2  511.48  5133.2   514.2    5154  516.49
  5196.9  520.26
#Mann= 3 , 1 , 0
 4865.70    0.13       0 4986.35    0.05       0  5013.8    0.13       0
Bank Sta=4986.35,5013.80
Exp/Cntr=0.3,0.1

Type RM Length L Ch R = 1 ,24489.8,524.8,524.8,524.8
XS GIS Cut Line= 3
      1893514.12       765839.15      1893722.00       765587.62
      1893920.49       765496.78
BEGIN DESCRIPTION:
South Fork 40.0
END DESCRIPTION:
#Sta/Elev= 30
  4673.7  520.44    4689  519.84  4705.2  518.98  4732.2   517.9  4744.7  516.97
  4765.2  515.92  4807.1  514.03  4822.5  513.05  4848.4  511.88  4868.8  510.69
  4889.8  509.08  4909.4  508.02  4971.4  504.29  4979.2  503.19  4986.2  501.27
  4989.2  497.27 5010.65  497.27 5013.65  501.27  5038.2   501.5  5043.7  502.06
  5055.3  504.05  5086.9  503.79  5100.9  504.01    5135  506.52  5148.2  508.41
  5152.6  509.14  5164.9  510.63  5176.7  512.46  5209.9  519.41  5218.3  520.89
#Mann= 3 , 1 , 0
 4673.70    0.11       0  4986.2    0.05       0 5013.65    0.13       0
Bank Sta=4986.20,5013.65
Exp/Cntr=0.3,0.1

Type RM Length L Ch R = 1 ,23965.0,556.7,556.7,556.7
XS GIS Cut Line= 3
      1893838.61       766182.51      1894118.75       765881.50
      1894186.14       765823.98
BEGIN DESCRIPTION:
South Fork 39.0
END DESCRIPTION:
#Sta/Elev= 30
  4588.8   520.3  4601.8  519.44  4622.2  517.82  4639.7  516.82  4643.1  516.44
  4648.8  515.49  4652.7  515.15  4689.3  513.06  4720.6  510.85  4749.7  509.09
  4764.3  508.01  4821.8  505.69  4872.7  504.02    4909  502.86  4929.1  502.65
  4933.1  502.25  4945.7  501.44  4971.7  499.97  4988.5  499.46    4991  495.46
 5008.88  495.46 5011.38  499.46  5013.2  499.57  5013.8  500.09  5018.5  506.58
  5026.8  508.54    5033  510.29  5046.5  515.01  5058.5  517.07  5088.6  521.79
#Mann= 3 , 1 , 0
 4588.80    0.11       0  4988.5    0.05       0 5011.38    0.13       0
Bank Sta=4988.50,5011.38
Exp/Cntr=0.3,0.1

Type RM Length L Ch R = 1 ,23408.3,754.8,754.8,754.8
XS GIS Cut Line= 3
      1894384.86       766350.21      1894432.12       766215.25
      1894477.04       766092.40
BEGIN DESCRIPTION:
South Fork 38.0
END DESCRIPTION:
#Sta/Elev= 29
    4857  517.29  4866.7  515.57  4880.6  513.68  4886.3  512.24  4900.9  509.47
  4912.3  507.78  4927.9  505.34  4940.2  503.61  4947.9  502.72  4953.1  502.28
  4965.5   501.5  4971.6  501.56  4978.4   501.5  4979.4  501.32  4986.2   499.1
  4989.2   495.1 5010.65   495.1 5013.65   499.1  5028.2  501.96  5029.6  502.49
  5045.5  504.26  5057.8  506.36  5072.5  508.36  5076.5  509.23  5085.7  510.47
  5094.4  511.83  5104.1  514.18  5116.2  516.43  5130.8   518.8
#Mann= 3 , 1 , 0
 4857.00    0.11       0  4986.2    0.05       0 5013.65    0.15       0
Bank Sta=4986.20,5013.65
Exp/Cntr=0.3,0.1

Type RM Length L Ch R = 1 ,22653.5,610,610,610
XS GIS Cut Line= 3
      1894564.29       766604.13      1894702.75       766653.81
      1894826.53       766692.43
BEGIN DESCRIPTION:
South Fork 37.0
END DESCRIPTION:
#Sta/Elev= 28
  4852.9  514.16  4861.6   513.3  4872.9  511.65  4878.3  510.77  4880.8  510.33
  4892.4  508.18  4911.6  505.39  4914.6  504.91  4918.3  504.09  4927.7  502.32
  4935.4  501.55  4961.6  499.45 4988.63  496.12 4991.13  492.12    5009  492.12
  5011.5  496.12    5014  496.52  5017.8  499.38  5020.3  501.02  5031.9  503.47
  5039.2  506.46  5052.2  510.62  5067.4  515.23    5068   515.4  5069.8  515.73
  5093.2  519.69  5098.5  520.22  5129.7  521.27
#Mann= 3 , 1 , 0
 4852.90    0.11       0 4988.63    0.05       0  5011.5    0.13       0
Bank Sta=4988.63,5011.50
Exp/Cntr=0.3,0.1

Type RM Length L Ch R = 1 ,22043.5,818.5,818.5,818.5
XS GIS Cut Line= 3
      1894230.09       767146.91      1894332.87       767134.88
      1894679.17       766972.19
BEGIN DESCRIPTION:
South Fork 36.0
END DESCRIPTION:
#Sta/Elev= 30
  4896.5     513  4903.3  511.29  4907.7  510.88  4934.1  504.07  4953.7  497.84
  4986.2  495.63  4989.2  491.63 5010.65  491.63 5013.65  495.63  5018.3  495.92
  5029.6  497.62  5051.6  498.54  5067.3  499.05  5098.6  499.44  5108.1  499.72
  5124.3  500.01  5141.2   500.5  5165.8  501.77  5181.2   502.7  5201.4  504.64
  5222.1  505.84  5235.1   506.9  5264.3  508.68    5287  509.83  5295.9   510.4
  5307.4  510.71  5341.9  512.17  5351.6  512.42  5375.5  513.64  5382.6  514.12
#Mann= 3 , 1 , 0
 4896.50    0.15       0  4986.2    0.05       0 5013.65    0.15       0
Bank Sta=4986.20,5013.65
Exp/Cntr=0.3,0.1

Type RM Length L Ch R = 1 ,21225.0,402.1,402.1,402.1
XS GIS Cut Line= 4
      1894674.96       767474.63      1894841.13       767374.12
      1894909.86       767335.66      1894898.40       767250.19
BEGIN DESCRIPTION:
South Fork 35.0
END DESCRIPTION:
#Sta/Elev= 30
  4805.8  507.08  4827.8  505.02  4841.8  503.35  4856.7  501.06  4876.1  498.93
  4890.2  497.56  4917.7  496.78  4925.1  496.06  4954.3  492.95  4967.3  492.27
 4988.63  492.18 4991.13  488.18 5008.88  488.18 5011.38  492.18    5024  495.42
  5024.3  495.14  5035.5  494.69    5055  497.44  5055.7  497.91  5057.6  497.99
  5078.8  498.07  5084.4  498.39  5089.1  498.55  5102.3  499.67  5107.4  499.99
  5130.4  503.95  5133.5  504.42  5143.3  505.47  5149.1  505.81    5165  507.31
#Mann= 3 , 1 , 0
 4805.80    0.13       0 4988.63    0.05       0 5011.38    0.15       0
Bank Sta=4988.63,5011.38
Exp/Cntr=0.3,0.1

Type RM Length L Ch R = 1 ,20822.9,650.5,650.5,650.5
XS GIS Cut Line= 3
      1894802.97       767656.73      1895174.25       767514.75
      1895231.89       767526.87
BEGIN DESCRIPTION:
South Fork 34.0
END DESCRIPTION:
#Sta/Elev= 30
  4602.5  507.13  4618.5  506.27  4632.8  505.75  4652.6  504.78  4674.9  504.07
  4703.9  503.36  4796.8     503  4812.5  503.18  4835.5  502.69  4850.7  501.22
  4865.9  500.78  4876.6  500.31  4885.6  499.35  4894.3  498.26  4910.4  495.82
  4935.9  493.26  4940.9  492.97  4961.5  491.32  4967.6  489.36  4972.8  488.24
  4984.7  488.12  4987.7  484.12  5012.3  484.12  5015.3  488.12  5025.6   493.1
  5026.2  493.01  5037.2  493.47    5042  498.79  5055.6  506.35  5058.9  507.36
#Mann= 3 , 1 , 0
 4602.50    0.12       0  4984.7    0.05       0  5015.3    0.15       0
Bank Sta=4984.70,5015.30
Exp/Cntr=0.3,0.1

Type RM Length L Ch R = 1 ,20172.4,534,534,534
XS GIS Cut Line= 3
      1894725.24       767800.10      1894847.25       767894.56
      1895096.65       768077.50
BEGIN DESCRIPTION:
South Fork 33.0
END DESCRIPTION:
#Sta/Elev= 29
  4845.7  504.55  4882.8  499.58  4891.4  498.58  4900.4  497.42  4908.8  495.59
  4913.5  494.69  4925.6  493.02  4936.2  491.98  4942.2  491.55  4959.4  490.66
  4984.7  487.05  4987.7  483.05  5012.3  483.05  5015.3  487.05  5016.6  487.31
  5016.9  487.29  5044.2  490.63  5050.4  490.82  5090.3  490.81  5152.1  491.77
  5185.1  492.58  5194.1  492.94    5227  494.62  5236.1  495.32  5253.9  496.28
    5269  497.61  5282.7  499.65  5293.6  501.95  5309.3  504.64
#Mann= 3 , 1 , 0
 4845.70    0.12       0  4984.7    0.05       0  5015.3    0.12       0
Bank Sta=4984.70,5015.30
Exp/Cntr=0.3,0.1

Type RM Length L Ch R = 1 ,19638.4,295.9,295.9,295.9
XS GIS Cut Line= 3
      1894425.18       768241.95      1894489.50       768280.12
      1894684.92       768397.58
BEGIN DESCRIPTION:
South Fork 32.0
END DESCRIPTION:
#Sta/Elev= 27
  4925.2  503.73    4928  502.86    4930  501.97  4942.4  495.53  4956.9  490.61
  4960.3  489.66 4981.98  484.09 4985.48  480.09 5014.53  480.09 5018.03  484.09
    5021  484.89    5026  487.65  5034.3  487.82  5063.5  488.73  5081.1  489.45
  5089.8  490.18  5095.7  490.96  5121.8  492.67  5123.1  492.82  5143.2  494.21
  5167.9  495.77  5178.9  497.45  5183.2  497.92  5188.5  498.72  5208.1  501.33
  5213.2  502.08    5228  503.56
#Mann= 3 , 1 , 0
 4925.20    0.13       0 4981.98    0.05       0 5018.03    0.13       0
Bank Sta=4981.98,5018.03
Exp/Cntr=0.3,0.1

Type RM Length L Ch R = 1 ,19342.5,737.3,737.3,737.3
XS GIS Cut Line= 3
      1894316.59       768542.63      1894447.73       768572.43
      1894635.60       768618.02
BEGIN DESCRIPTION:
South Fork 31.0
END DESCRIPTION:
#Sta/Elev= 30
  4862.2  503.56  4876.1  500.88  4879.5  500.39  4895.4  496.79  4902.4  493.64
  4908.1  492.52  4923.4  490.79  4942.6   488.9  4947.7  488.18  4953.2  487.69
  4968.3  482.66  4968.8  482.37 4987.13  481.92 4989.63  477.92  5010.5  477.92
    5013  481.92  5024.2  487.01  5024.6  487.31  5045.5  488.25  5065.8  489.02
  5082.6  489.97  5098.9  491.38  5113.1  492.81    5126  495.01  5128.8  495.58
  5142.7   496.9  5152.8  498.09  5171.2  500.61  5176.7  501.26    5190  503.06
#Mann= 3 , 1 , 0
 4862.20    0.12       0 4987.13    0.05       0    5013    0.12       0
Bank Sta=4987.13,5013.00
Exp/Cntr=0.3,0.1

Type RM Length L Ch R = 1 ,18605.2,804.4,804.4,804.4
XS GIS Cut Line= 4
      1894296.89       769190.09      1894324.25       769102.25
      1894380.03       768955.24      1894713.48       768730.77
BEGIN DESCRIPTION:
South Fork 30.0
END DESCRIPTION:
#Sta/Elev= 30
    4908  511.26  4914.8  510.27  4924.1  508.22  4929.4  506.31  4941.4  500.47
  4949.3  495.89  4959.7  491.37  4963.9  488.65  4978.1  484.89  4983.4  483.74
  4986.1  481.78  4988.8  477.78 5011.34  477.78 5014.04  481.78  5028.8  483.44
    5036  483.77  5057.4  486.65  5078.1  488.29  5098.6  489.55  5139.3  494.84
  5161.8  495.64  5201.9  498.69  5237.6  501.74  5254.6   502.9  5292.9   504.4
  5376.1  505.97  5406.6  507.38  5443.4  508.35  5478.9  508.64  5559.2  511.63
#Mann= 3 , 1 , 0
 4908.00    0.13       0  4986.1    0.05       0 5014.04    0.13       0
Bank Sta=4986.10,5014.04
Exp/Cntr=0.3,0.1

Type RM Length L Ch R = 1 ,17800.8,489.5,489.5,489.5
XS GIS Cut Line= 3
      1894770.41       769273.03      1894873.37       769239.81
      1894955.21       769222.21
BEGIN DESCRIPTION:
South Fork 29.0
END DESCRIPTION:
#Sta/Elev= 22
  4891.8   498.4  4900.9  496.25  4914.4  493.43  4926.9  490.74  4952.1  486.42
    4954  486.13  4954.4  486.03  4955.4  485.89 4987.13  480.05 4989.63  476.05
  5010.5  476.05    5013  480.05  5013.4   480.2    5014   480.3  5021.6  482.84
  5032.5  483.39  5043.9  485.26  5055.7  489.62  5060.1  490.39  5063.3  491.86
  5067.6  493.57  5083.7  498.83
#Mann= 3 , 1 , 0
 4891.80    0.13       0 4987.13    0.05       0    5013    0.15       0
Bank Sta=4987.13,5013.00
Exp/Cntr=0.3,0.1

Type RM Length L Ch R = 1 ,17311.3,484.3,484.3,484.3
XS GIS Cut Line= 3
      1894770.50       769620.46      1894881.00       769725.12
      1894967.43       769803.98
BEGIN DESCRIPTION:
South Fork 28.0
END DESCRIPTION:
#Sta/Elev= 30
  4847.8   495.8  4865.6  493.38    4868  492.95  4884.6  490.53  4888.2  489.35
  4896.6  487.34  4908.1  485.39  4920.7  483.41  4927.7  482.63  4939.3  481.72
  4946.7  480.94  4970.6  478.75  4988.3   477.7  4988.8  477.65  4989.6  477.38
  4991.6  473.38  5008.3  473.38  5010.3  477.38  5012.1  477.69  5012.9  477.62
  5021.7  479.96  5025.6  480.38    5037   482.9  5047.5  485.27  5066.1  489.91
  5082.9  492.25  5087.6  492.74  5103.2  493.88  5109.5  494.55    5117  495.16
#Mann= 3 , 1 , 0
 4847.80    0.14       0  4989.6    0.05       0  5010.3    0.15       0
Bank Sta=4989.60,5010.30
Exp/Cntr=0.3,0.1

Type RM Length L Ch R = 1 ,16827.0,852.6,852.6,852.6
XS GIS Cut Line= 3
      1894590.03       770107.84      1894645.65       770108.89
      1894782.58       770022.19
BEGIN DESCRIPTION:
South Fork 27.0
END DESCRIPTION:
#Sta/Elev= 27
  4943.8  491.96    4959  486.07  4972.7  480.83  4986.8  474.32    4987   474.3
  4989.5   470.3 5010.38   470.3 5012.88   474.3  5021.7  474.78  5027.5  474.32
  5033.4  474.34  5039.5  475.36  5040.6  475.62  5041.5  475.81  5051.3  477.24
  5067.8   479.4    5071  479.64  5075.8  480.01  5098.6  482.22  5101.3  482.71
  5107.8  483.61  5117.6   485.1  5123.5  485.93  5139.4  487.77  5141.8  488.01
  5145.4  488.42  5161.5  490.13
#Mann= 3 , 1 , 0
 4943.80    0.15       0    4987    0.05       0 5012.88    0.15       0
Bank Sta=4987.00,5012.88
Exp/Cntr=0.3,0.1

Type RM Length L Ch R = 1 ,15974.4,421.4,421.4,421.4
XS GIS Cut Line= 3
      1894938.64       770345.69      1895312.32       770218.27
      1895465.05       770065.54
BEGIN DESCRIPTION:
South Fork 26.0
END DESCRIPTION:
#Sta/Elev= 30
  4601.5  488.08  4625.8  487.25    4638  486.45  4651.5  484.97  4663.2  484.63
  4678.7  483.37  4707.8  482.77  4720.6  479.98  4762.4  477.96  4789.4  474.77
  4811.6  474.09  4825.7  473.12  4855.3  471.72  4896.4  471.19  4928.9  471.68
  4945.6  472.76  4973.7  470.54 4987.13   470.2 4989.63   466.2 5010.38   466.2
 5012.88   470.2  5014.7  471.46  5023.6  473.21  5055.9  474.15  5071.8  475.32
  5093.6  474.81  5107.4  475.05  5143.3  478.24  5188.3  485.04  5212.3  487.42
#Mann= 3 , 1 , 0
 4601.50    0.15       0 4987.13    0.05       0 5012.88    0.15       0
Bank Sta=4987.13,5012.88
Exp/Cntr=0.3,0.1

Type RM Length L Ch R = 1 ,15553.0,551.7,551.7,551.7
XS GIS Cut Line= 3
      1894980.58       770415.33      1895119.61       770463.06
      1895181.31       770525.53
BEGIN DESCRIPTION:
South Fork 25.0
END DESCRIPTION:
#Sta/Elev= 21
  4855.4  485.33  4871.1  484.06  4890.2  481.91  4904.3  477.56  4909.9  475.69
  4920.4   472.4  4933.8  472.22  4959.5  471.02 4985.58  468.86 4988.38  464.86
 5011.62  464.86 5014.42  468.86  5015.7   470.3  5024.7  471.57  5028.8  472.55
  5044.3  474.83  5046.3  475.03  5067.9  481.58  5069.6  481.97  5078.1   483.6
  5090.2  486.97
#Mann= 3 , 1 , 0
 4855.40    0.15       0 4985.58    0.05       0 5014.42    0.15       0
Bank Sta=4985.58,5014.42
Exp/Cntr=0.3,0.1

Type RM Length L Ch R = 1 ,15001.3,613.2,613.2,613.2
XS GIS Cut Line= 3
      1894660.30       770926.50      1894830.10       770868.52
      1894985.71       770832.47
BEGIN DESCRIPTION:
South Fork 24.0
END DESCRIPTION:
#Sta/Elev= 30
  4820.5  492.25  4823.4  492.35  4834.7  491.99  4848.4  490.89  4864.4  489.96
  4884.8  486.73  4911.3  484.56  4920.7  482.89  4939.9  478.87  4941.7  477.96
  4942.8  477.72  4961.5  465.41  4983.5  465.48  4989.6  465.05  4991.6  461.05
  5008.3  461.05  5010.3  465.05  5015.3   469.1    5033  469.05  5037.4  469.12
  5053.3  469.82  5073.7  471.56  5090.3  473.53  5093.6  474.16  5099.3  474.71
  5114.8  477.19  5131.8  479.79  5135.6  480.57  5152.2  484.95  5159.7  485.71
#Mann= 3 , 1 , 0
 4820.50    0.15       0  4989.6    0.05       0  5010.3    0.14       0
Bank Sta=4989.60,5010.30
Exp/Cntr=0.3,0.1

Type RM Length L Ch R = 1 ,14388.1,986.9,986.9,986.9
XS GIS Cut Line= 4
      1894727.21       771665.14      1894722.85       771527.01
      1895114.50       771395.00      1895164.05       771398.85
BEGIN DESCRIPTION:
South Fork 23.0
END DESCRIPTION:
#Sta/Elev= 30
  4448.5  486.66  4463.1  482.52  4472.4  482.68  4490.9  483.76  4502.7  482.94
  4552.3  481.82  4586.7  479.92  4622.4  479.24    4649   479.7  4659.8  479.54
  4672.4  478.86  4694.9  478.48  4725.9  477.42  4733.2  476.89  4765.1  475.58
  4783.6  474.61  4813.1   472.4  4831.3  471.89  4889.3  467.62  4915.6  466.84
  4933.5  466.57  4951.8  466.76  4956.9  465.49    4982  461.49  4984.5  457.49
 5015.63  457.49 5018.13  461.49  5027.8  466.16  5037.5  479.87  5049.7  488.43
#Mann= 3 , 1 , 0
 4448.50    0.12       0    4982    0.05       0 5018.13    0.13       0
Bank Sta=4982.00,5018.13
Exp/Cntr=0.3,0.1

Type RM Length L Ch R = 1 ,13401.2,413.1,413.1,413.1
XS GIS Cut Line= 3
      1894927.48       772116.78      1895014.52       772079.10
      1895255.64       771931.60
BEGIN DESCRIPTION:
South Fork 22.0
END DESCRIPTION:
#Sta/Elev= 29
  4906.3  480.58  4922.9   475.4  4931.4  471.16  4946.8  468.14    4951  467.15
  4976.4  460.52  4980.6   459.5 4984.16  459.36 4986.36  455.36 5013.75  455.36
 5015.95  459.36  5018.4  462.92  5023.8  465.98  5033.7  466.65  5050.9  468.12
  5064.5  469.08  5068.4  469.29  5104.7  472.12  5125.7  473.19  5137.6  474.06
  5154.9  475.87  5160.2  476.29  5167.6  477.08  5177.7  477.68  5199.6  479.31
  5242.3  480.13  5255.6  480.67    5277  481.71  5283.8  482.44
#Mann= 3 , 1 , 0
 4906.30    0.13       0 4984.16    0.05       0 5015.95    0.11       0
Bank Sta=4984.16,5015.95
Exp/Cntr=0.3,0.1

Type RM Length L Ch R = 1 ,12988.1,500.7,500.7,500.7
XS GIS Cut Line= 3
      1895173.76       772487.58      1895216.50       772430.63
      1895395.41       772216.68
BEGIN DESCRIPTION:
South Fork 21.0
END DESCRIPTION:
#Sta/Elev= 27
  4928.8  482.59  4933.8  479.61    4951  477.02  4954.6  475.15  4972.6  466.22
  4972.8  466.19    4982  459.35  4984.5  455.35  5015.5  455.35    5018  459.35
  5031.2  463.66  5043.4  467.25  5069.4  468.05    5077  469.17  5082.7  469.78
  5103.7  471.12  5123.2  471.68  5137.1  471.71  5153.3  472.41  5203.9  475.52
  5223.2  477.03  5224.9  477.33  5237.1  478.55  5248.3  479.34  5255.1  480.24
  5262.3  480.88  5278.9  482.08
#Mann= 3 , 1 , 0
 4928.80    0.11       0    4982    0.05       0    5018    0.11       0
Bank Sta=4982.00,5018.00
Exp/Cntr=0.3,0.1

Type RM Length L Ch R = 1 ,12487.4,564.9,564.9,564.9
XS GIS Cut Line= 4
      1895694.08       772633.62      1895754.10       772537.43
      1895715.04       772399.41      1895648.67       772226.11
BEGIN DESCRIPTION:
South Fork 20.0
END DESCRIPTION:
#Sta/Elev= 30
  4738.9  481.25  4775.8   478.3  4783.8  477.19  4793.8  475.61  4833.1  471.74
  4841.8  470.96    4902  467.51  4905.4  467.29  4911.4  466.61  4943.3  465.47
  4962.6  464.22    4980  463.23  4981.8  462.53    4984  459.33 4984.05  459.34
 4986.25  455.34 5013.64  455.34 5015.84  459.34  5026.9  462.93  5049.9  465.93
  5051.1  466.17  5067.9  466.77  5105.1  469.84  5119.7  471.46    5131  473.48
  5141.1  474.71    5147  475.58  5156.6  477.86  5164.3   479.1  5181.3  481.19
#Mann= 3 , 1 , 0
 4738.90    0.11       0 4984.05    0.05       0 5015.84    0.11       0
Bank Sta=4984.05,5015.84
Exp/Cntr=0.3,0.1

Type RM Length L Ch R = 1 ,11922.5,500,500,500
XS GIS Cut Line= 3
      1895868.47       772741.21      1896257.72       772303.46
      1896301.09       772191.34
BEGIN DESCRIPTION:
South Fork 19.0
END DESCRIPTION:
#Sta/Elev= 30
  4414.2  480.93  4460.5  476.52  4478.3   475.3  4508.1     474  4527.5   472.8
  4540.9  472.32  4548.9  471.76  4574.1  471.02  4657.4     468    4696  467.88
  4723.7  467.08  4756.9  466.44    4771  466.36    4784  465.81    4801  464.61
  4830.1   465.2  4864.7  465.45  4883.6  465.91  4921.8  465.64  4958.6  464.41
  4969.9  461.24  4985.6   459.8  4987.6   455.8  5012.5   455.8  5014.5   459.8
  5038.5  460.12  5072.1  470.15  5088.5  476.34  5118.7  480.26  5120.2   480.6
#Mann= 3 , 1 , 0
 4414.20    0.11       0  4985.6    0.05       0  5014.5    0.11       0
Bank Sta=4985.60,5014.50
Exp/Cntr=0.3,0.1

Type RM Length L Ch R = 1 ,11422.5,530.5,530.5,530.5
XS GIS Cut Line= 3
      1896106.64       772919.76      1896689.00       772498.37
      1896769.00       772389.67
BEGIN DESCRIPTION:
South Fork 18.0
END DESCRIPTION:
#Sta/Elev= 30
  4277.2  479.42  4306.4  476.56  4332.9  475.42  4348.1  474.14  4391.5  472.07
  4430.3  470.74  4466.9  469.75  4532.7   468.3  4621.1  465.11  4645.8  464.76
  4696.4  464.72  4731.4  464.38  4802.4  464.32  4848.2  463.79  4873.1  463.95
  4922.5  464.92  4951.7  464.91  4969.3  464.39  4983.3  463.82  4985.6  458.22
  4987.6  454.22  5012.5  454.22  5014.5  458.22  5019.3  462.63  5085.6  465.64
  5100.5  476.16  5110.9  487.27  5113.9  488.45  5126.8  494.14    5131  494.33
#Mann= 3 , 1 , 0
 4277.20    0.11       0  4985.6    0.05       0  5014.5    0.11       0
Bank Sta=4985.60,5014.50
Exp/Cntr=0.3,0.1

Type RM Length L Ch R = 1 ,10892.0,494,494,494
XS GIS Cut Line= 3
      1896897.40       773090.89      1897093.63       772829.19
      1897102.34       772630.48
BEGIN DESCRIPTION:
South Fork 17.0
END DESCRIPTION:
#Sta/Elev= 30
  4672.9  476.96  4684.1   475.9    4707  474.33  4726.4  472.79  4732.5   472.2
  4752.6  469.85  4757.9  469.32    4770  468.97  4814.4   466.4  4833.6   465.5
  4864.9  464.47  4932.7  462.78  4946.4  463.26  4964.2  463.46  4978.4  456.97
  4981.4  452.97 5018.75  452.97 5021.75  456.97  5035.3  461.79  5040.2  462.97
    5060  463.03  5076.3  462.72  5110.7  462.69  5130.6  462.81  5153.4  463.34
  5164.2  463.95  5173.4  465.83  5181.5  467.17  5184.1   468.4  5198.9  478.21
#Mann= 3 , 1 , 0
 4672.90    0.11       0  4978.4    0.05       0 5021.75    0.11       0
Bank Sta=4978.40,5021.75
Exp/Cntr=0.3,0.1

Type RM Length L Ch R = 1 ,10398.0,528.2,528.2,528.2
XS GIS Cut Line= 3
      1896986.18       773176.98      1897422.50       772916.81
      1897670.47       772808.43
BEGIN DESCRIPTION:
South Fork 16.0
END DESCRIPTION:
#Sta/Elev= 30
    4492  480.52  4519.1  474.02  4537.9  471.98    4547  470.36  4571.6   467.8
  4593.2  466.34  4604.7  464.91  4625.6  463.69  4641.6  463.02  4728.6  462.24
  4774.9  462.06  4844.9  462.35  4866.9  462.24  4906.8  461.25  4939.6  461.39
 4977.35  456.16 4980.35  452.16  5019.5  452.16  5022.5  456.16  5025.4  458.56
  5043.2  461.55  5058.1  461.94  5075.7  462.85  5101.5  466.07  5124.8  468.32
  5159.9  468.75  5179.7  468.64  5205.3  469.24  5228.1  469.23  5270.6  470.18
#Mann= 3 , 1 , 0
 4492.00    0.11       0 4977.35    0.05       0  5022.5    0.11       0
Bank Sta=4977.35,5022.50
Exp/Cntr=0.3,0.1

Type RM Length L Ch R = 1 ,9869.8,577.4,577.4,577.4
XS GIS Cut Line= 3
      1897222.93       773386.24      1897344.95       773407.38
      1897751.20       772821.45
BEGIN DESCRIPTION:
South Fork 15.0
END DESCRIPTION:
#Sta/Elev= 30
  4823.4  476.66  4838.9  475.07  4864.8  470.96  4899.2  464.07  4925.6  461.36
  4947.3  459.78  4969.4  459.21    4985     454    4987     450  5013.1     450
  5015.1     454  5016.8  454.22  5032.6  460.35  5047.3  460.31  5075.2  461.85
  5150.3  462.66  5187.5  462.27  5223.9  462.66  5265.7  462.17  5284.6   461.4
  5301.2  460.09  5323.4   459.9    5402  460.74  5425.2  461.66  5447.1  463.08
  5491.6  467.89  5529.8  470.75  5543.6  471.41  5580.3  471.79  5660.3  471.55
#Mann= 3 , 1 , 0
 4823.40    0.11       0    4985    0.05       0  5015.1    0.11       0
Bank Sta=4985.00,5015.10
Exp/Cntr=0.5,0.3

Type RM Length L Ch R = 1 ,9292.4,48,48,48
XS GIS Cut Line= 5
      1897616.36       773530.07      1897769.28       773410.96
      1897857.51       773171.27      1897934.16       772824.03
      1897977.49       772836.78
BEGIN DESCRIPTION:
Upstream Section of Bridge/Culvert/Weir
END DESCRIPTION:
#Sta/Elev= 27
  4551.9  476.23  4874.9  470.15  4886.2  469.92  4899.8  469.43  4927.1  467.57
    4936  467.23  4944.7   466.3 4965.25   456.9 4968.75     450 5031.25     450
 5034.63   456.9  5052.4  457.44  5053.8  457.59  5058.1  457.73  5066.4  459.26
  5098.5  460.43  5112.8  460.66  5126.9  463.41  5133.5  463.94    5141  465.34
  5157.9  467.14  5174.6  469.24  5198.3  470.08    5242  470.37  5254.6  470.58
  5261.5   470.8  5401.9   473.5
#Mann= 3 , 1 , 0
 4551.90    0.11       0 4965.25    0.05       0 5034.63    0.11       0
#XS Ineff= 2 , 0
       0    4915   468.5    5083       0   468.5
Bank Sta=4965.25,5034.63
Exp/Cntr=0.5,0.3

Type RM Length L Ch R = 3 ,9268.4,,,
BEGIN DESCRIPTION:
South Fork - Lindley Rd
Structure ID: NCF-0100
Approximate Survey Structure
END DESCRIPTION:
Bridge Culvert--1,0,-1,-1, 0
Deck Dist Width WeirC Skew NumUp NumDn MinLoCord MaxHiCord MaxSubmerge Is_Ogee
10,28,2.6,, 28, 28,,,0.95,0,1,1,,
  4551.9  4604.4  4606.5  4631.6  4874.9  4886.2  4899.8 4927.41  4927.5 5072.39
  5072.5  5098.5  5112.8  5119.2  5123.1  5126.9  5133.5    5141  5157.9  5166.2
  5174.6  5179.5  5198.3  5237.3  5240.2  5254.6  5264.3  5401.9
  476.23  475.42  475.27  474.74  470.16  469.93   469.7   469.7   469.7   469.7
   469.7   469.7   469.7   469.7     470  470.05   470.1  470.16  470.28  470.34
  470.62  470.78  471.12  471.36  471.53  471.98  472.29   473.5
  476.23  475.24   475.2  474.73  470.15  469.92  469.43  467.56   467.7   467.7
  459.48  460.43  460.66  461.91  462.67  463.41  463.94  465.34  467.14  468.18
  469.24  469.41  470.08  470.34  470.36  470.58  470.83   473.5
  4551.9  4604.4  4606.5  4631.6  4874.9  4886.2  4899.8 4927.41  4927.5 5072.39
  5072.5  5098.5  5112.8  5119.2  5123.1  5126.9  5133.5    5141  5157.9  5166.2
  5174.6  5179.5  5198.3  5237.3  5240.2  5254.6  5264.3  5401.9
  476.23  475.42  475.27  474.74  470.16  469.93   469.7   469.7   469.7   469.7
   469.7   469.7   469.7   469.7     470  470.05   470.1  470.16  470.28  470.34
  470.62  470.78  471.12  471.36  471.53  471.98  472.29   473.5
  475.98  474.99  474.95  474.48   469.9  469.67  469.18  467.31  467.45  467.45
  459.23  460.18  460.41  461.66  462.42  463.16  463.69  465.09  466.89  467.93
  468.99  469.16  469.83  470.09  470.11  470.33  470.58  473.25
Pier Skew, UpSta & Num, DnSta & Num=,4951.7, 2 ,4951.7, 2 , 0 , 0 , 0 ,,
       1       1
  461.87   468.7
       1       1
  461.62  468.45
Pier Skew, UpSta & Num, DnSta & Num=,5000.0, 2 ,5000.0, 2 , 0 , 0 , 0 ,,
       1       1
     449   468.7
       1       1
  448.75  468.45
Pier Skew, UpSta & Num, DnSta & Num=,5048.4, 2 ,5048.4, 2 , 0 , 0 , 0 ,,
       1       1
   456.3   468.7
       1       1
  456.05  468.45
BR Coef= 1 , 1 , 0 ,1.25, 0 ,,,0.8,0,2,0,
Wspro=,,,, 1 ,,,, 0 ,,,, 0 ,,,,-1 ,-1 ,-1 , 0 , 0 , 0 , 0 , 0
BC Design=,, 0 ,, 0 ,,,,,,
BR U #Sta/Elev= 82
  4551.9  476.23  4556.8  476.14  4559.6  476.09  4560.9  476.06  4564.2     476
  4604.4  475.24  4606.5   475.2  4631.6  474.73  4650.6  474.37  4658.3  474.23
  4666.6  474.07  4678.9  473.84  4680.8   473.8    4681   473.8  4681.2   473.8
  4689.5  473.64  4705.4  473.34  4711.1  473.23  4714.4  473.17  4719.2  473.08
  4727.1  472.93  4728.7   472.9  4745.3  472.59  4745.7  472.58  4750.6  472.49
  4752.9  472.45  4768.1  472.16  4785.6  471.83  4797.3  471.61  4802.6  471.51
  4819.2   471.2  4820.8  471.17  4823.7  471.11  4836.5  470.87  4874.9  470.15
  4875.3  470.14  4886.2  469.92  4899.8  469.43  4927.1  467.57 4927.41  467.56
  4927.5  467.55  4927.6  467.55    4936  467.23  4944.7   466.3 4965.25   456.9
 4968.75     450    5000     450 5031.25     450 5034.63   456.9  5052.4  457.44
  5053.8  457.59  5058.1  457.73  5066.4  459.26  5072.3  459.48 5072.39  459.48
  5072.5  459.48  5098.5  460.43  5108.7  460.62  5112.8  460.66  5119.2  461.91
  5123.1  462.67  5125.3   463.1  5126.9  463.41  5131.1  463.79  5133.5  463.94
    5141  465.34  5157.9  467.14  5166.2  468.18  5174.6  469.24  5179.5  469.41
  5182.1  469.51  5197.8  470.06  5198.3  470.08  5199.5   470.1  5237.3  470.34
  5240.2  470.36    5242  470.37  5254.6  470.58  5261.5   470.8  5263.5  470.81
  5264.3  470.83  5401.9   473.5
BR U #Mann= 3
 4551.90    0.11 4965.25    0.05 5034.63    0.11
BR U Banks=4965.25,5034.63
BR D #Sta/Elev= 82
  4551.9  475.98  4556.8  475.89  4559.6  475.84  4560.9  475.81  4564.2  475.75
  4604.4  474.99  4606.5  474.95  4631.6  474.48  4650.6  474.12  4658.3  473.98
  4666.6  473.82  4678.9  473.59  4680.8  473.55    4681  473.55  4681.2  473.55
  4689.5  473.39  4705.4  473.09  4711.1  472.98  4714.4  472.92  4719.2  472.83
  4727.1  472.68  4728.7  472.65  4745.3  472.34  4745.7  472.33  4750.6  472.24
  4752.9   472.2  4768.1  471.91  4785.6  471.58  4797.3  471.36  4802.6  471.26
  4819.2  470.95  4820.8  470.92  4823.7  470.86  4836.5  470.62  4874.9   469.9
  4875.3  469.89  4886.2  469.67  4899.8  469.18  4927.1  467.32 4927.41  467.31
  4927.5   467.3  4927.6   467.3    4936  466.98  4944.7  466.05 4965.25  456.65
 4968.75  449.75    5000  449.75 5031.25  449.75 5034.63  456.65  5052.4  457.19
  5053.8  457.34  5058.1  457.48  5066.4  459.01  5072.3  459.23 5072.39  459.23
  5072.5  459.23  5098.5  460.18  5108.7  460.37  5112.8  460.41  5119.2  461.66
  5123.1  462.42  5125.3  462.85  5126.9  463.16  5131.1  463.54  5133.5  463.69
    5141  465.09  5157.9  466.89  5166.2  467.93  5174.6  468.99  5179.5  469.16
  5182.1  469.26  5197.8  469.81  5198.3  469.83  5199.5  469.85  5237.3  470.09
  5240.2  470.11    5242  470.12  5254.6  470.33  5261.5  470.55  5263.5  470.56
  5264.3  470.58  5401.9  473.25
BR D #Mann= 3
 4551.90    0.11 4965.25    0.05 5034.63    0.11
BR D Banks=4965.25,5034.63

Type RM Length L Ch R = 1 ,9244.4,597.7,597.7,597.7
XS GIS Cut Line= 5
      1897656.70       773504.07      1897809.62       773384.96
      1897897.85       773145.27      1897974.50       772798.03
      1898017.83       772810.77
BEGIN DESCRIPTION:
Downstream Section of Bridge/Culvert/Weir
END DESCRIPTION:
#Sta/Elev= 27
  4551.9  475.98  4874.9   469.9  4886.2  469.67  4899.8  469.18  4927.1  467.32
    4936  466.98  4944.7  466.05 4965.25  456.65 4968.75  449.75 5031.25  449.75
 5034.63  456.65  5052.4  457.19  5053.8  457.34  5058.1  457.48  5066.4  459.01
  5098.5  460.18  5112.8  460.41  5126.9  463.16  5133.5  463.69    5141  465.09
  5157.9  466.89  5174.6  468.99  5198.3  469.83    5242  470.12  5254.6  470.33
  5261.5  470.55  5401.9  473.25
#Mann= 3 , 1 , 0
 4551.90    0.11       0 4965.25    0.05       0 5034.63    0.11       0
#XS Ineff= 2 , 0
       0    4915   468.5    5083       0   468.5
Bank Sta=4965.25,5034.63
Exp/Cntr=0.5,0.3

Type RM Length L Ch R = 1 ,8646.7,809.8,809.8,809.8
XS GIS Cut Line= 4
      1897798.84       773472.64      1897897.63       773481.62
      1898154.13       773453.84      1898183.91       773440.09
BEGIN DESCRIPTION:
South Fork 14.0
END DESCRIPTION:
#Sta/Elev= 30
  4900.8  470.66  4909.5  470.08  4918.7  468.74  4923.8  467.75  4944.7  465.46
  4949.1  464.39  4950.2  464.92  4956.9  462.41  4965.7  460.83  4980.5  453.83
    4983  449.83 5016.88  449.83 5019.38  453.83    5033  456.76  5053.4  457.51
  5084.6  457.63  5104.7  458.63  5124.1  460.24  5133.2  462.76  5152.2  464.71
  5179.4  463.74  5182.8  463.43  5190.1  461.85  5198.2     464  5217.3  466.98
  5221.7   468.3  5236.4  469.14  5254.5  471.65  5267.4  473.98  5290.8  475.66
#Mann= 4 , 1 , 0
 4900.80    0.13       0  4980.5    0.05       0 5019.38    0.13       0
  5152.2      10       0
Bank Sta=4980.50,5019.38
Exp/Cntr=0.3,0.1

Type RM Length L Ch R = 1 ,7836.9,465.1,465.1,465.1
XS GIS Cut Line= 3
      1898365.02       774044.46      1898352.86       773849.79
      1898413.72       773606.34
BEGIN DESCRIPTION:
South Fork 13.0
END DESCRIPTION:
#Sta/Elev= 30
  4796.8  472.45  4802.8  470.93  4812.9  469.63  4820.7  468.34  4839.6  466.12
  4916.7  459.28  4935.4  458.03  4971.6  456.38  4979.3  452.02  4984.4  451.17
  4986.4  447.17  5013.6  447.17  5015.6  451.17  5024.7  454.45  5033.1  456.53
  5045.6  457.27  5076.7   458.4  5097.7  458.84    5117   458.9  5134.9  458.72
  5155.5  458.69  5170.3  458.88  5183.4  459.59  5188.1  460.03  5201.3  460.71
  5206.2  460.82  5212.4  464.18  5223.8  470.01  5237.8  471.08  5242.8  471.34
#Mann= 3 , 1 , 0
 4796.80    0.15       0  4984.4    0.05       0  5015.6    0.13       0
Bank Sta=4984.40,5015.60
Exp/Cntr=0.3,0.1

Type RM Length L Ch R = 1 ,7371.8,481.6,481.6,481.6
XS GIS Cut Line= 3
      1898587.61       774042.19      1898813.62       773794.37
      1898850.11       773755.12
BEGIN DESCRIPTION:
South Fork 12.0
END DESCRIPTION:
#Sta/Elev= 29
  4664.6  470.02  4669.7  469.84  4683.7  469.19  4702.3  467.99  4724.3  466.82
  4727.5  466.59  4734.8  466.12  4745.9  465.34  4751.8  464.99    4780  462.35
  4802.8  461.19  4807.4  460.73  4834.9   458.6  4846.7  457.55  4890.3  455.63
  4924.4  455.08    4965  454.98  4969.2  454.63  4971.5  454.25  4973.4  453.18
  4984.5  448.98  4986.5  444.98  5013.6  444.98  5015.6  448.98  5025.7  456.36
  5026.6  456.84  5027.4   457.4  5028.9  457.98  5053.6  471.15
#Mann= 3 , 1 , 0
 4664.60    0.15       0  4984.5    0.05       0  5015.6    0.15       0
Bank Sta=4984.50,5015.60
Exp/Cntr=0.3,0.1

Type RM Length L Ch R = 1 ,6890.2,427.1,427.1,427.1
XS GIS Cut Line= 3
      1899033.73       774221.17      1899112.63       774157.62
      1899276.94       774081.00
BEGIN DESCRIPTION:
South Fork 11.0
END DESCRIPTION:
#Sta/Elev= 28
  4898.7  470.82  4912.1  467.76  4924.2  466.89  4929.7  465.86  4933.1   465.1
  4940.9  462.02  4952.2  459.22  4961.2  456.84  4964.8  456.38  4973.1  453.57
  4979.8  447.63 4980.63  447.63 4983.13  443.63    5017  443.63  5019.5  447.63
  5041.1  450.67  5042.9  451.24  5057.8  451.83  5076.6  455.42  5086.2  455.56
  5110.4   456.7  5133.1  461.67    5137   462.3  5139.8  463.23  5147.9  464.93
  5167.2  468.04  5174.6  469.03  5181.3  470.28
#Mann= 3 , 1 , 0
 4898.70    0.15       0 4980.63    0.05       0  5019.5    0.15       0
Bank Sta=4980.63,5019.50
Exp/Cntr=0.3,0.1

Type RM Length L Ch R = 1 ,6463.1,420.6,420.6,420.6
XS GIS Cut Line= 3
      1899133.34       774464.57      1899436.19       774426.18
      1899506.89       774387.43
BEGIN DESCRIPTION:
South Fork 10.0
END DESCRIPTION:
#Sta/Elev= 30
  4693.7  467.35    4729  461.98  4741.5  460.27    4757  460.45  4776.3  459.19
  4790.2   459.1  4798.5  459.17  4808.4  458.86  4811.4  458.87  4837.3  456.59
  4850.4  456.29  4856.9   455.9  4876.3  455.26  4879.6   454.5  4903.3     453
  4907.9  452.89  4921.7  453.78  4929.9  454.17  4937.4  454.29  4955.9  450.25
    4974   449.4 4986.05  447.62 4987.85  443.62 5012.24  443.62 5014.04  447.62
  5017.3   450.9  5028.8  456.99    5046  462.03  5064.7  465.91  5079.6  470.84
#Mann= 3 , 1 , 0
 4693.70    0.15       0 4986.05    0.05       0 5014.04    0.15       0
Bank Sta=4986.05,5014.04
Exp/Cntr=0.3,0.1

Type RM Length L Ch R = 1 ,6042.5,572,572,572
XS GIS Cut Line= 4
      1899382.31       774923.59      1899623.69       774867.16
      1899710.49       774745.63      1899771.37       774661.23
BEGIN DESCRIPTION:
South Fork 9.0
END DESCRIPTION:
#Sta/Elev= 30
  4599.8  467.28    4607  466.26  4623.3   463.5  4630.2  462.83  4639.9  462.06
  4650.3  461.56  4666.8  459.99  4701.8  457.45  4719.6  455.16  4753.5   453.4
  4766.6  453.31  4796.4  453.54  4812.6  454.08  4852.8  454.84  4859.3  454.67
  4919.7  455.41  4932.1  455.31  4950.9  454.48  4961.1  453.71  4984.4  446.71
  4986.4  442.71  5013.5  442.71  5015.5  446.71  5018.2   447.6  5027.6  452.69
    5041  454.28    5065  458.45  5074.9  460.48  5091.8  465.51  5101.1   467.9
#Mann= 3 , 1 , 0
 4599.80    0.15       0  4984.4    0.05       0  5015.5    0.15       0
Bank Sta=4984.40,5015.50
Exp/Cntr=0.3,0.1

Type RM Length L Ch R = 1 ,5470.5,493.5,493.5,493.5
XS GIS Cut Line= 3
      1899871.84       775356.02      1899934.62       775252.94
      1899899.32       774757.89
BEGIN DESCRIPTION:
South Fork 8.0
END DESCRIPTION:
#Sta/Elev= 30
  4879.3  465.79  4890.5  462.56  4900.8  458.06  4905.5  454.82  4914.7  451.76
  4942.4  452.15  4967.7  452.18  4976.3   449.7  4980.5  446.66    4983  442.66
 5016.88  442.66 5019.38  446.66  5027.8  449.74  5032.1  451.91  5033.8  452.27
  5049.1  452.06  5065.4  452.15  5103.6  452.79  5132.7  452.75  5142.8  451.87
  5164.5  452.49  5177.1  452.47  5182.3  452.64    5225  455.66  5253.3   456.8
  5351.9  462.08    5353   462.1  5354.4  461.73    5361  461.76  5496.3  463.99
#Mann= 3 , 1 , 0
 4879.30    0.15       0  4980.5    0.05       0 5019.38    0.14       0
Bank Sta=4980.50,5019.38
Exp/Cntr=0.3,0.1

Type RM Length L Ch R = 1 ,4977.0,1086.6,1086.6,1086.6
XS GIS Cut Line= 3
      1900426.96       775204.24      1900277.87       774964.63
      1900056.37       774618.08
BEGIN DESCRIPTION:
South Fork 7.0
END DESCRIPTION:
#Sta/Elev= 30
  4717.8   465.6  4738.2   463.6  4750.3     462  4779.6  458.84  4784.4  458.62
  4798.5   457.2  4808.4  455.39  4843.6  451.08  4863.3   449.8  4886.7  449.23
  4957.9  450.48  4975.1  447.53  4980.5  445.01    4983  441.01 5016.88  441.01
 5019.38  445.01  5039.1  445.39  5071.5  448.34  5077.9  448.72  5090.2   448.8
  5107.9  449.78    5141  449.94  5208.6  449.41    5237  449.61  5254.5  449.35
  5299.4  449.63  5338.6  450.47  5378.9  452.75  5391.8  452.95  5411.3  461.57
#Mann= 3 , 1 , 0
 4717.80    0.14       0  4980.5    0.05       0 5019.38    0.13       0
Bank Sta=4980.50,5019.38
Exp/Cntr=0.3,0.1

Type RM Length L Ch R = 1 ,3890.4,506.5,506.5,506.5
XS GIS Cut Line= 4
      1900442.89       775168.53      1900338.97       774978.27
      1900717.87       774507.00      1900771.84       774440.16
BEGIN DESCRIPTION:
South Fork 6.0
END DESCRIPTION:
#Sta/Elev= 30
  4178.5  463.28    4210  458.32    4252  452.85  4275.9  450.66  4292.6  450.06
  4363.8  449.47  4395.3  449.78  4459.2  449.41  4513.6  449.49  4558.8  450.12
  4651.5  449.64  4705.4   449.9  4711.6  449.64  4757.1  449.46  4811.7  449.78
  4838.5  449.52  4873.2  448.54  4896.2  448.23  4911.3  448.65  4936.7  448.27
  4976.2  448.34  4984.5  442.38  4986.5  438.38  5013.6  438.38  5015.6  442.38
  5026.8  445.23  5035.9  448.41  5050.8  458.51    5057  460.65  5085.9   463.8
#Mann= 3 , 1 , 0
 4178.50    0.12       0  4984.5    0.05       0  5015.6    0.15       0
Bank Sta=4984.50,5015.60
Exp/Cntr=0.3,0.1

Type RM Length L Ch R = 1 ,3383.9,610.5,610.5,610.5
XS GIS Cut Line= 3
      1900633.62       775354.19      1901128.00       774765.69
      1901273.90       774587.24
BEGIN DESCRIPTION:
South Fork 5.0
END DESCRIPTION:
#Sta/Elev= 30
  4231.4  465.73  4251.9  459.49  4277.7  457.75  4292.3  455.35  4328.6  451.53
  4387.3  448.92  4428.5  449.29  4558.9  447.65  4623.4  448.04  4655.8  451.38
  4671.1  454.47  4691.9  455.83  4715.8     456  4791.7  450.35  4850.7  447.87
  4880.6  447.13  4940.3  447.01  4975.6  447.63  4984.4  441.02  4986.4  437.02
  5013.6  437.02  5015.6  441.02  5032.4  447.02  5096.7  446.56  5145.9  447.68
  5182.3  449.98  5196.9  452.01  5205.7  456.75  5225.9  464.18  5230.5  464.94
#Mann= 4 , 1 , 0
 4231.40      10       0  4715.8    0.13       0  4984.4    0.05       0
  5015.6    0.15       0
Bank Sta=4984.40,5015.60
Exp/Cntr=0.3,0.1

Type RM Length L Ch R = 1 ,2773.4,878.4,878.4,878.4
XS GIS Cut Line= 4
      1901292.28       775212.64      1901298.16       775207.87
      1901587.12       775079.19      1901668.73       775047.05
BEGIN DESCRIPTION:
South Fork 4.0
END DESCRIPTION:
#Sta/Elev= 30
  4676.1  463.05  4719.9  462.87    4740   462.3  4754.5  461.07  4772.1   460.1
  4785.2  458.54  4812.4  457.54  4818.1  456.87  4837.9  455.61  4840.2  455.35
  4847.1  453.57  4850.2  453.09  4876.3  450.05  4898.6  445.07  4905.6  444.58
  4925.9  444.32  4934.7  443.89  4951.6   444.3  4961.1  443.67  4988.3  438.31
  4989.8  434.31 5010.13  434.31 5011.63  438.31  5015.7  445.77  5028.6   446.5
  5043.8  448.48  5061.2  453.05  5072.5  457.85  5075.8  458.67  5087.7  460.08
#Mann= 3 , 1 , 0
 4676.10    0.13       0  4988.3    0.05       0 5011.63    0.15       0
Bank Sta=4988.30,5011.63
Exp/Cntr=0.3,0.1

Type RM Length L Ch R = 1 ,1895.0,718,718,718
XS GIS Cut Line= 3
      1901441.46       776058.34      1901695.63       775891.56
      1901944.19       775759.00
BEGIN DESCRIPTION:
South Fork 3.0
END DESCRIPTION:
#Sta/Elev= 30
    4696  460.56  4698.4  460.22  4710.5  453.35  4712.6  452.45  4725.8  448.42
  4735.4   447.4  4765.6  445.78  4782.2  444.47  4799.2  443.81  4905.7  443.34
  4941.4   443.8  4959.1  443.76  4973.8  441.32  4984.4  436.67  4986.4  432.67
  5013.6  432.67  5015.6  436.67  5042.5  443.23  5052.2  447.97  5087.1  448.71
  5096.1  449.38  5171.9  453.21  5194.6  453.65  5201.4  453.46  5215.9  453.65
  5231.8  454.26  5248.2  455.36  5261.4   456.8  5266.9  457.98  5281.7     460
#Mann= 3 , 1 , 0
 4696.00    0.15       0  4984.4    0.05       0  5015.6    0.15       0
Bank Sta=4984.40,5015.60
Exp/Cntr=0.3,0.1

Type RM Length L Ch R = 1 ,1177.0,649.7,649.7,649.7
XS GIS Cut Line= 3
      1901630.70       776511.81      1901758.50       776497.50
      1902253.47       776124.46
BEGIN DESCRIPTION:
South Fork 2.0
END DESCRIPTION:
#Sta/Elev= 30
  4871.4  462.77  4883.4  456.33  4890.1  452.03  4892.8  450.88  4916.5   446.2
  4932.9   444.7  4938.6   443.2    4968   439.2 4987.52  435.82 4989.12  431.82
 5010.88  431.82 5012.48  435.82  5015.9  439.13  5028.6  442.44  5068.7  442.02
  5104.8  442.86  5170.3  445.55  5224.9  445.99    5246  445.45    5272   445.3
  5328.3  445.87  5407.4  444.66  5466.1  444.49  5513.6  444.85  5536.3  445.64
  5557.6  447.16    5562  448.06  5580.1  450.09  5593.6   453.7  5619.8  459.88
#Mann= 4 , 1 , 0
 4871.40    0.15       0 4987.52    0.05       0 5012.48    0.11       0
  5224.9      10       0
Bank Sta=4987.52,5012.48
Exp/Cntr=0.3,0.1

Type RM Length L Ch R = 1 ,527.3,0,0,0
XS GIS Cut Line= 4
      1901659.46       776612.13      1902267.44       776668.50
      1902268.37       776434.69      1902282.98       776131.94
BEGIN DESCRIPTION:
South Fork 1.0
END DESCRIPTION:
#Sta/Elev= 30
  4155.6  460.58    4166   458.6  4180.8   456.6  4202.6  454.99  4215.1  452.89
  4243.8  450.53  4276.9  449.13  4298.8  448.67  4338.3  448.79  4371.5  448.13
  4471.5  448.82  4525.6  448.05  4820.6  446.87  4841.4  445.18  4851.2  445.44
  4865.6  443.48  4900.2  441.46  4933.3     442  4976.6  434.53  4979.6  430.53
  5020.4  430.53  5023.4  434.53  5035.2  444.66  5201.3  445.23  5223.8  447.42
  5231.6  449.11  5251.9  451.87  5271.6  455.21  5287.7   458.7  5303.1  461.41
#Mann= 3 , 1 , 0
 4155.60    0.13       0  4976.6   0.045       0  5023.4    0.11       0
Bank Sta=4976.60,5023.40
Exp/Cntr=0.3,0.1

Chan Stop Cuts=-1
